--- SFKCHERRYRV.prj (project) ---

Proj Title=SFKCHERRYRV
Current Plan=p01
Default Exp/Contr=0,0
English Units
Geom File=g01
Flow File=f01
Plan File=p01
Background Map Layer=stream
BEGIN DESCRIPTION:
Stream Name- South Fork Cherry River
Flood Zone: Zone A
Greenbrier County, WV
County-Wide Study
WVDHSEM-2018-3, Flood Risk Project
HEC-RAS Version: 5.0.7
General Notes:
For the Hydrology Regression was used.
END DESCRIPTION:
DSS Export Rating Curves= 0
DSS Export Rating Curve Sorted= 0
DSS Export Volume Flow Curves= 0
DXF Filename=..\..\..\..\Users\pratik.pathak\Desktop\DisasterStudies\ModelsCherry\SFKCHERRYRV\SFKCHERRYRV.
DXF OffsetX= 0
DXF OffsetY= 0
DXF ScaleX= 0
DXF ScaleY= 0

--- SFKCHERRYRV.p01 (plan) ---

Plan Title=Floodplain
Program Version=5.07
Short Identifier=Floodplain
Geom File=g01
Flow File=f01
Subcritical Flow
K Sum by GR= 0
Std Step Tol= 0.01
Critical Tol= 0.01
Num of Std Step Trials= 20
Max Error Tol= 0.3
Flow Tol Ratio= 0.001
Split Flow NTrial= 30
Split Flow Tol= 0.02
Split Flow Ratio= 0.02
Log Output Level= 0
Friction Slope Method= 1
Unsteady Friction Slope Method= 2
Unsteady Bridges Friction Slope Method= 1
Parabolic Critical Depth
Global Vel Dist= 0 , 0 , 0
Global Log Level= 0
CheckData=True
Encroach Param=-1 ,0,0, 0
Computation Interval=0.1SEC
Output Interval=1MIN
Instantaneous Interval=Max Profile
Mapping Interval=1HOUR
Computation Time Step Use Courant=        0
Computation Time Step Use Time Series=    0
Computation Time Step Count To Double=0
Computation Time Step Max Doubling=0
Computation Time Step Max Halving=0
Computation Time Step Residence Courant=0
Run HTab= 0
Run UNet= 0
Run Sediment= 0
Run PostProcess= 0
Run WQNet= 0
Run RASMapper= 0
UNET Theta= 0
UNET Theta Warmup= 0
UNET ZTol= 0
UNET ZSATol= 0
UNET MxIter= 0
UNET Max Iter WO Improvement= 0
UNET MaxInSteps= 0
UNET DtIC= 0
UNET DtMin= 0
UNET MaxCRTS= 0
UNET WFStab= 0
UNET SFStab= 0
UNET WFX= 1
UNET SFX= 1
UNET 1D Methodology=Finite Difference
UNET DSS MLevel= 1
UNET Pardiso=0
UNET DZMax Abort= 0
UNET Use Existing IB Tables= 0
UNET Froude Reduction=False
UNET Froude Limit= 0
UNET Froude Power= 0
UNET D1 Cores= 0
UNET D2 Coriolis=0
UNET D2 Cores= 0
UNET D2 Theta= 1
UNET D2 Theta Warmup= 1
UNET D2 Z Tol= 0.01
UNET D2 Volume Tol= 0.01
UNET D2 Max Iterations= 20
UNET D2 Equation= 0
UNET D2 RampUpFraction=0.1
UNET D2 TimeSlices= 1
UNET D2 BCVolumeCheck=0
UNET D1D2 MaxIter= 0
UNET D1D2 ZTol=0.01
UNET D1D2 QTol=0.1
UNET D1D2 MinQTol=1
DSS File=dss
Write IC File= 0
Write IC File at Fixed DateTime=0
Write IC File at Sim End=0
Echo Input=False
Echo Parameters=False
Echo Output=False
Write Detailed= 0
HDF Write Warmup=0
HDF Write Time Slices=0
HDF Flush=0
HDF Face Node Velocities=0
HDF Compression= 1
HDF Chunk Size= 1
HDF Spatial Parts= 1
HDF Use Max Rows=0
HDF Fixed Rows= 1
Calibration Method= 0
Calibration Iterations= 20
Calibration Max Change=0.05
Calibration Tolerance=0.2
Calibration Maximum=1.5
Calibration Minimum=0.5
Calibration Optimization Method= 1
WQ AD Non Conservative
WQ ULTIMATE=-1
WQ Max Comp Step=1HOUR
WQ Output Interval=15MIN
WQ Output Selected Increments= 0
WQ Output face flow=0
WQ Output face velocity=0
WQ Output face area=0
WQ Output face dispersion=0
WQ Output cell volume=0
WQ Output cell surface area=0
WQ Output cell continuity=0
WQ Output cumulative cell continuity=0
WQ Output face conc=0
WQ Output face dconc_dx=0
WQ Output face courant=0
WQ Output face peclet=0
WQ Output face adv mass=0
WQ Output face disp mass=0
WQ Output cell mass=0
WQ Output cell source sink temp=0
WQ Output nsm pathways=0
WQ Output nsm derived pathways=0
WQ Output MaxMinRange=-1
WQ Daily Max Min Mean=-1
WQ Daily Range=0
WQ Daily Time=0
WQ Create Restart=0
WQ Fixed Restart=0
WQ System Summary=0
WQ Write To DSS=0
WQ Use Fixed Temperature=0
Sorting and Armoring Iterations= 10
XS Update Threshold= 0.02
Bed Roughness Predictor= 0
Hydraulics Update Threshold= 0.02
Energy Slope Method= 1
Volume Change Method= 1
Sediment Retention Method= 0
XS Weighting Method= 0
Number of US Weighted Cross Sections= 1
Number of DS Weighted Cross Sections= 1
Upstream XS Weight=0
Main XS Weight=1
Downstream XS Weight=0
Number of DS XS's Weighted with US Boundary= 1
Upstream Boundary Weight= 1
Weight of XSs Associated with US Boundary= 0
Number of US XS's Weighted with DS Boundary= 1
Downstream Boundary Weight= 0.5
Weight of XSs Associated with DS Boundary= 0.5
Percentile Method= 0
Sediment Output Level= 3
Mass or Volume Output= 0
Output Increment Type= 1
Profile and TS Output Increment= 1
XS Output Flag= 0
XS Output Increment= 10
Write Gradation File= 0
Read Gradation Hotstart= 0
Write HDF5 File= 1
Write Binary Output= 1
Write DSS Sediment File= 0
SV Curve= 0
Specific Gage Flag= 0

--- SFKCHERRYRV.f01 (steady flow) ---

Flow Title=NFF Regression Equation
Program Version=5.07
Number of Profiles= 6
Profile Names=f1p,f10p,f4p,f2p,f02p,f1pplus
River Rch & RM=SFKCHERRYRV,Main            ,78918
     522     275     366     442     731     773
River Rch & RM=SFKCHERRYRV,Main            ,77950
     600     317     422     508     837     887
River Rch & RM=SFKCHERRYRV,Main            ,76458
     671     357     473     569     935     993
River Rch & RM=SFKCHERRYRV,Main            ,75421
     750     401     530     637    1040    1110
River Rch & RM=SFKCHERRYRV,Main            ,73155
     834     447     591     709    1160    1230
River Rch & RM=SFKCHERRYRV,Main            ,70251
    1020     551     725     868    1410    1510
River Rch & RM=SFKCHERRYRV,Main            ,68863
    1130     615     808     966    1560    1680
River Rch & RM=SFKCHERRYRV,Main            ,63626
    1380     755     988    1180    1900    2040
River Rch & RM=SFKCHERRYRV,Main            ,62089
    1530     842    1100    1310    2100    2270
River Rch & RM=SFKCHERRYRV,Main            ,58079
    1810     998    1300    1550    2470    2670
River Rch & RM=SFKCHERRYRV,Main            ,53834
    3210    1810    2340    2760    4340    4750
River Rch & RM=SFKCHERRYRV,Main            ,46931
    4030    2290    2940    3470    5420    5950
River Rch & RM=SFKCHERRYRV,Main            ,37279
    5180    2980    3810    4470    6950    7670
River Rch & RM=SFKCHERRYRV,Main            ,31911
    5860    3390    4320    5060    7840    8670
River Rch & RM=SFKCHERRYRV,Main            ,19173
    6560    3810    4840    5670    8750    9700
Boundary for River Rch & Prof#=SFKCHERRYRV,Main            , 1
Up Type= 0
Dn Type= 1
Dn Known WS=2239
Boundary for River Rch & Prof#=SFKCHERRYRV,Main            , 2
Up Type= 0
Dn Type= 1
Dn Known WS=2236
Boundary for River Rch & Prof#=SFKCHERRYRV,Main            , 3
Up Type= 0
Dn Type= 1
Dn Known WS=2237
Boundary for River Rch & Prof#=SFKCHERRYRV,Main            , 4
Up Type= 0
Dn Type= 1
Dn Known WS=2238
Boundary for River Rch & Prof#=SFKCHERRYRV,Main            , 5
Up Type= 0
Dn Type= 1
Dn Known WS=2241
Boundary for River Rch & Prof#=SFKCHERRYRV,Main            , 6
Up Type= 0
Dn Type= 1
Dn Known WS=2242.5
DSS Import GetInterval= 0
DSS Import GetPeak= 0
DSS Import FillOption= 0

--- SFKCHERRYRV.g01 (geometry) ---

Geom Title=USGS 10m DEM
Program Version=5.07

River Reach=SFKCHERRYRV     ,Main
Reach XY= 30
2145838.48200002420658.6550000012143387.57230879420086.037806675
2141698.41936006414709.8745444862139156.30250002412673.142500013
2136758.31834434412549.8237722962132873.67999999415120.391000018
2131836.71681154414266.2515992672129428.13500001414699.322999999
2128482.06199999416763.2370000032126626.20201254417473.214039296
2125150.18000004419254.3490000222126013.56000002422259.320999995
2127199.07300001422662.1050000042127293.41900003424285.692000002
2126229.05451368424947.7218344662126437.33499999426507.665999994
2125173.62900002428373.8860000072122125.03300002429433.327000022
 2121193.4787035430869.2930150182121387.75299999433125.912000015
2122722.87841745435414.660688221     2122237.936436307.703000009
2123208.09600522437710.5964638292122021.18900003439457.042000011
2119706.14300005439804.028000012    2114906.4465443943.471500024
2113418.52800001442606.1560000032111659.08300003442217.361000016
2108560.76700002443938.5470000062106032.08700004444387.307999998

Type RM Length L Ch R = 1 ,78918   ,131.2,131.6,131.2
XS GIS Cut Line= 2
     2145811.294      420280.274     2145786.572      421082.368
#Sta/Elev= 30
       0 3641.18    32.8 3627.58    42.6 3621.86    55.7 3617.66    98.3 3599.58
   114.6 3586.57     131 3585.94   137.6 3583.65   150.7 3573.07   163.8 3567.97
   193.2 3548.52   209.6 3544.54   252.2 3521.34   268.6 3516.21   317.7    3511
   337.4 3500.26   353.7 3487.31   360.3 3484.97   373.4  3483.7   386.5 3485.16
   406.2 3488.73     452 3490.37     488 3493.84   520.8 3506.56   537.2 3510.81
   648.5 3530.75   700.9  3538.1   779.6  3561.3   792.6 3563.43   802.5 3567.57
#Mann= 3 ,-1 , 0
       0     .12       0   360.3     .04       0   386.5     .12       0
Bank Sta=360.3,386.5
XS Rating Curve= 0 ,0
Exp/Cntr=0.3,0.1

Type RM Length L Ch R = 1 ,78786   ,109.2,108.3,107.4
XS GIS Cut Line= 2
2145665.64995532420285.1273474782145670.53133075420939.231655003
#Sta/Elev= 30
       0 3618.36    35.6 3601.81    53.5 3595.81    68.4 3588.23    78.3 3579.98
   104.5 3578.69   114.3  3571.7   137.3  3562.7   150.4 3555.04   163.6 3549.77
   183.2 3537.64   199.6  3530.5   209.5 3528.61   222.6 3530.96   229.2 3530.21
   242.3 3524.21     272 3516.13   288.2 3508.85   304.6 3497.02   330.9 3482.85
   347.3 3480.46   379.5 3479.62   383.4 3479.14   390.6 3479.69   397.2 3481.86
   423.7 3496.53   435.9 3500.32     531 3511.98   570.4 3514.79   654.1 3528.85
#Mann= 3 , 0 , 0
       0     .12       0   379.5     .04       0   390.6     .12       0
Bank Sta=379.5,390.6
XS Rating Curve= 0 ,0
Exp/Cntr(USF)=0,0
Exp/Cntr=0.3,0.1

Type RM Length L Ch R = 1 ,78678   ,186.4,186.6,188.3
XS GIS Cut Line= 3
2145542.63929451 420322.225800742145563.14107131420718.593485599
2145610.97855052420888.465350539
#Sta/Elev= 30
       0 3581.49     8.4 3580.46    18.2 3575.48    47.8 3574.56    57.6 3571.12
    67.5    3562    86.6  3554.8    97.1 3548.56   106.9 3539.72   142.8 3516.99
     166 3498.96   181.4 3489.18   202.2 3478.77   215.3 3476.04   225.2 3477.21
   251.5  3476.4   317.2 3478.95   333.9 3477.13   343.4 3476.47     350 3477.43
   363.2 3487.23   376.3 3492.96   392.8  3494.2   423.2 3500.11   457.1 3504.65
   478.4 3507.03   491.4 3506.97   505.1 3508.23   544.9 3513.01   573.4 3517.58
#Mann= 3 , 0 , 0
       0     .12       0   333.9     .04       0     350     .12       0
Bank Sta=333.9,350
XS Rating Curve= 0 ,0
Exp/Cntr(USF)=0,0
Exp/Cntr=0.3,0.1

Type RM Length L Ch R = 1 ,78491   ,242,234.8,226.4
XS GIS Cut Line= 3
2145409.86588283420330.0360014272145459.65591221420693.210333367
2145503.58829107420921.658703458
#Sta/Elev= 30
       0 3578.92     7.2 3572.45    30.3 3571.18    40.3 3563.31    50.2 3560.36
    60.1 3553.98    73.4 3549.13    86.6 3541.95   121.7 3514.67   136.3 3506.86
   159.5 3490.22   176.1 3472.61   206.2 3471.35   212.5 3470.89   217.9 3471.37
   232.4 3473.87     282 3473.92     292 3477.31   305.2 3479.56   331.7  3479.2
   354.9 3489.07   361.5 3490.75   408.2 3490.15   418.2 3494.39   430.8 3496.97
   447.6 3495.95   461.7  3496.9   501.8 3506.43   541.9 3510.85   599.2 3523.07
#Mann= 3 , 0 , 0
       0     .12       0   206.2     .04       0   217.9     .12       0
#XS Ineff= 2 , 0
                          257.33         3479.08
Permanent Ineff=
       F       F
Bank Sta=206.2,217.9
XS Rating Curve= 0 ,0
Exp/Cntr(USF)=0,0
Exp/Cntr=0.3,0.1

Type RM Length L Ch R = 1 ,78256   ,167.9,182,197.9
XS GIS Cut Line= 4
      2145204.23      420252.805     2145267.408       420664.84
     2145363.549      420777.462     2145396.512      420977.986
#Sta/Elev= 30
       0 3609.14    32.6 3594.97    42.3 3589.46    52.1 3587.14    84.7 3575.61
    94.4 3569.31   120.5 3567.13   133.5 3560.03   208.4 3531.47   231.2 3524.92
   270.3 3510.95   319.2 3498.86   348.5 3480.82   364.7 3467.82     381 3463.76
     394 3465.83   416.8 3464.15   455.5 3467.11   475.7  3464.8   490.7 3464.41
   500.6 3466.62   513.4 3481.47   519.9 3484.65   561.7 3488.69     578 3494.44
   587.9 3493.72   630.5 3498.14   689.5 3511.55   722.3 3515.45   768.1 3526.58
#Mann= 3 , 0 , 0
       0     .12       0   475.7     .04       0   490.7     .12       0
Bank Sta=475.7,490.7
XS Rating Curve= 0 ,0
Exp/Cntr=0.3,0.1

Type RM Length L Ch R = 1 ,78074   ,130.1,124.2,122
XS GIS Cut Line= 4
 2145135.5325837420333.9411017712145185.32261308420598.511650038
2145156.03436051420758.6207641192145167.74966154420939.231655003
#Sta/Elev= 30
       0 3571.74     3.2 3569.43     6.6 3568.79    26.6 3568.63    36.6 3563.24
      60 3555.29   103.4 3537.08   130.1 3528.63   160.2 3515.82   186.9 3508.76
   210.2 3500.77   230.3 3497.23     253 3490.63     267 3482.61   290.3 3462.19
   293.7 3459.99   325.53459.363     337 3459.12     347 3459.38     357 3460.75
     367 3460.33   383.7 3465.13   410.9 3476.06   432.5 3482.18   466.6 3486.08
   501.6 3492.91   548.8 3498.56   570.9 3499.88   584.9 3503.28     613 3507.57
#Mann= 3 , 0 , 0
       0     .12       0   325.5     .04       0     347     .12       0
Bank Sta=325.5,347
XS Rating Curve= 0 ,0
Exp/Cntr(USF)=0,0
Exp/Cntr=0.3,0.1

Type RM Length L Ch R = 1 ,77950   ,227.3,226.1,223.9
XS GIS Cut Line= 3
2145048.62544022420298.9055282092145059.84367466420588.977018808
2145058.24106974420952.768335746
#Sta/Elev= 30
       0 3591.15    21.8 3581.34      35 3569.94      58 3567.78    74.4 3556.39
    87.5 3553.93    94.1 3550.45   103.9 3547.87   120.3  3541.7   143.1 3530.73
   159.7 3526.26   169.6 3520.58   212.3 3508.44   235.3 3499.67   261.5 3492.27
   274.7 3485.02   283.1  3478.1   305.3 3463.43   323.9 3456.89   333.7 3451.45
   340.3  3450.8   351.5 3451.41   392.8 3456.26   402.6  3461.2     419 3472.52
   432.1  3479.3   560.1 3490.52     606 3500.88   632.3 3508.46   654.1 3517.39
#Mann= 3 , 0 , 0
       0     .12       0   333.7     .04       0   351.5     .12       0
Bank Sta=333.7,351.5
XS Rating Curve= 0 ,0
Exp/Cntr(USF)=0,0
Exp/Cntr=0.3,0.1

Type RM Length L Ch R = 1 ,77724   ,318.1,321.6,334.7
XS GIS Cut Line= 2
     2144808.676      420288.515     2144860.867      420966.998
#Sta/Elev= 30
       0 3590.37    26.2 3579.57    42.5 3574.16    68.7 3561.17    91.6 3560.01
   101.4 3552.78   111.2 3547.48   140.7  3533.4   160.3 3526.44     193 3509.61
   206.1 3506.44   232.3  3496.2   281.4 3481.59   304.3 3469.89   330.4 3447.27
   338.3 3443.23   346.8  3442.6   359.9 3443.33   369.7 3447.37     386 3449.54
   431.8 3447.54   438.4 3449.19   448.2  3455.7   474.4 3458.74   497.3 3469.83
   539.8 3482.77   552.9 3488.99   608.5 3509.04   660.9 3530.02   680.5 3536.28
#Mann= 3 ,-1 , 0
       0     .12       0   338.3     .04       0   359.9     .12       0
Bank Sta=338.3,359.9
XS Rating Curve= 0 ,0
Exp/Cntr=0.3,0.1

Type RM Length L Ch R = 1 ,77402   ,171,170.2,171.6
XS GIS Cut Line= 2
2144629.01854872420306.4931962652144429.94355405420843.239700882
#Sta/Elev= 30
       0 3564.81     8.2 3561.41    22.2 3549.34    25.7 3548.31    45.2 3548.04
    50.2 3546.78    74.7 3528.69    99.2 3515.86   116.6 3503.91   134.2 3496.51
   148.2 3487.71   172.6 3477.05   197.1 3469.15   216.2 3466.79   221.3  3465.1
   228.6 3459.64   235.6 3451.57   253.1 3434.81     257 3432.57   260.1 3432.07
   274.9 3432.46   308.1 3432.68   333.6 3437.19   346.4 3437.94   361.7 3443.04
   396.6 3458.27   417.6  3458.5   445.6 3461.25   561.1  3481.4   572.5 3484.24
#Mann= 3 , 0 , 0
       0     .12       0     257     .04       0   274.9     .12       0
Bank Sta=257,274.9
XS Rating Curve= 0 ,0
Exp/Cntr(USF)=0,0
Exp/Cntr=0.3,0.1

Type RM Length L Ch R = 1 ,77232   ,192.4,193.1,195.1
XS GIS Cut Line= 2
 2144467.6426379420294.3224981242144254.35646448420804.431929538
#Sta/Elev= 30
       0 3537.14    18.1 3537.38    28.1 3534.74    39.3 3525.67    50.7 3520.73
    71.3 3509.76    78.4  3507.7   106.9 3490.48   117.5 3486.99   142.4 3474.24
   153.1 3472.12   163.8 3466.96   173.6 3459.32   196.1  3439.4     210 3430.31
   224.2 3425.49   237.6 3424.07   248.8 3423.66   253.8 3424.22   270.4 3431.52
   281.1 3431.07   291.8 3432.77   299.1 3435.31   333.1 3451.12   341.6 3453.83
     370 3458.57   455.4 3467.03   479.5 3474.34     498 3477.29   552.9 3492.12
#Mann= 3 , 0 , 0
       0     .12       0   237.6     .04       0   253.8     .12       0
Bank Sta=237.6,253.8
XS Rating Curve= 0 ,0
Exp/Cntr(USF)=0,0
Exp/Cntr=0.3,0.1

Type RM Length L Ch R = 1 ,77039   ,189.8,188.7,187.8
XS GIS Cut Line= 2
2144333.36330407420180.2300159682144029.94157771420760.187999282
#Sta/Elev= 30
       0 3537.96    25.3 3523.58    46.3 3523.46    62.3 3516.05    91.9 3509.19
   106.7 3507.57   162.3  3490.5   177.1 3482.83   209.2 3455.84   228.9 3435.92
   247.4 3421.94   256.5 3417.57   262.7 3416.97   274.73417.543   288.2 3418.17
   299.3 3422.69   310.4 3421.67   328.9 3424.95   347.4 3424.54   376.8 3429.07
   398.8 3441.34   402.9 3442.34   458.5 3449.13   475.9 3449.64   510.3 3455.74
   537.4 3455.81   556.8 3458.14     577 3470.44   610.3 3482.67   654.5 3496.36
#Mann= 3 , 0 , 0
       0     .12       0   256.5     .04       0   274.7     .12       0
Bank Sta=256.5,274.7
XS Rating Curve= 0 ,0
Exp/Cntr(USF)=0,0
Exp/Cntr=0.3,0.1

Type RM Length L Ch R = 1 ,76851   ,235,237.1,238.2
XS GIS Cut Line= 2
2144126.38476043  420139.69002242143886.43781534420703.120997166
#Sta/Elev= 30
       0 3500.43    14.9 3490.09    29.2 3485.55      47 3477.45   100.9 3463.42
   143.3 3450.95   168.4 3433.97   178.9 3425.08   189.6 3417.92   203.9 3416.16
   213.4 3417.39   220.9 3416.72   246.7 3410.83   250.3 3410.61   265.9 3411.05
   285.9 3421.25   293.1 3421.98   307.3  3426.3   338.5 3428.79   357.2 3433.58
   403.6 3436.57     421 3434.63   433.5  3437.8   478.6  3439.1   503.5 3441.67
   523.5 3449.08     532 3453.79   542.7 3456.83   553.5 3463.52   612.4  3488.8
#Mann= 3 , 0 , 0
       0     .12       0   246.7     .04       0   265.9     .12       0
Bank Sta=246.7,265.9
XS Rating Curve= 0 ,0
Exp/Cntr(USF)=0,0
Exp/Cntr=0.3,0.1

Type RM Length L Ch R = 1 ,76613   ,155.6,155.3,138.2
XS GIS Cut Line= 3
2143986.42927996419966.6585380552143749.36585312420389.249864164
2143638.04911356 420642.80465983
#Sta/Elev= 30
       03511.979  26.0353504.772  32.3273501.254  44.3763492.013  63.6553491.875
  67.4153489.811  74.9383483.287  93.7473473.215 135.1273455.028 165.222 3446.43
 195.3163443.641  244.223432.721 271.5413410.868 278.0763407.515 285.3673405.813
 304.4093404.012 319.1063405.532 334.5033409.788 368.3593411.367 379.6453414.562
 413.5013420.542 459.3043426.027 510.0363441.065 535.2163451.288 599.614 3466.99
 656.9433476.725 674.6533481.935 682.3463482.653 735.7713496.128 761.4583503.678
#Mann= 3 , 0 , 0
       0     .12       0 285.367     .04       0 319.106     .12       0
Bank Sta=285.367,319.106
XS Rating Curve= 0 ,0
Exp/Cntr=0.3,0.1

Type RM Length L Ch R = 1 ,76458   ,125.3,125.1,131.7
XS GIS Cut Line= 4
2143867.89565082419871.522583257 2143705.7510245 420155.69357784
2143692.37827181420332.8825509342143617.15653795420598.666010574
#Sta/Elev= 30
       0 3505.35    15.7 3497.46    34.3 3486.08      56 3484.24    75.2 3472.75
   109.2 3457.09   203.7 3423.71   271.7 3421.23   310.9 3417.82   328.2 3413.87
   351.2 3402.08   357.8 3400.51   380.8 3398.99   413.7 3397.59   422.8 3398.46
     440 3399.14   449.9 3404.27   456.6 3406.01   476.2  3417.4   489.4 3422.98
   526.6 3430.87   551.4 3441.32   570.7 3444.97   635.4 3461.97   656.8 3465.18
     707 3476.06   727.5 3481.66   737.7 3486.13     765 3491.75   781.1 3496.77
#Mann= 3 ,-1 , 0
       0     .12       0   380.8     .04       0   422.8     .12       0
Bank Sta=380.8,422.8
XS Rating Curve= 0 ,0
Exp/Cntr=0.3,0.1

Type RM Length L Ch R = 1 ,76333   ,123.1,125.7,140
XS GIS Cut Line= 4
2143812.26712197419884.9195105192143614.95586966420116.865184778
2143553.03372132420307.8792694622143459.62573486420500.992410021
#Sta/Elev= 30
       0 3483.22     7.5 3481.45    20.8 3473.69    55.3 3460.91    81.1 3449.28
   151.9  3424.1   194.5 3416.71   249.6 3412.66   296.2 3406.98   322.2 3400.42
   346.4 3401.36     360 3396.86   380.9 3396.12   398.1 3388.49     415 3387.88
   429.2 3388.56   442.9 3392.19   453.3 3397.95   467.1 3402.49     474 3407.89
   484.3 3418.75     505 3429.02   553.5  3445.3     567 3448.14   596.1 3458.05
     618    3463   647.1 3473.34   666.5 3478.14   704.2 3492.85   719.8 3501.61
#Mann= 3 , 0 , 0
       0     .12       0   398.1     .04       0   429.2     .12       0
Bank Sta=398.1,429.2
XS Rating Curve= 0 ,0
Exp/Cntr(USF)=0,0
Exp/Cntr=0.3,0.1

Type RM Length L Ch R = 1 ,76207   ,127.4,127.2,130.7
XS GIS Cut Line= 2
     2143855.503      419810.555     2143218.223      420398.391
#Sta/Elev= 30
       0 3520.27    26.2  3504.5    55.6 3492.23    68.7 3482.58    94.9 3479.48
   111.2 3469.75     157 3452.27   219.2 3421.38   261.7 3413.85   327.2 3409.24
   359.9 3403.66   428.6 3403.31   448.2 3392.53   500.6 3385.82   513.6 3379.77
   516.9 3379.13   536.6 3379.63   559.5 3381.41   585.6  3390.4   608.5 3394.07
   644.5 3419.34   667.4 3432.76   680.5 3437.41   703.4 3449.74   732.8 3469.98
   755.8 3483.38   775.4 3486.04     795 3498.63   817.9 3507.46     867 3530.98
#Mann= 3 , 0 , 0
       0     .12       0   513.6     .04       0   536.6     .12       0
Bank Sta=513.6,536.6
XS Rating Curve= 0 ,0
Exp/Cntr=0.3,0.1

Type RM Length L Ch R = 1 ,76080   ,293.4,293.2,309.8
XS GIS Cut Line= 2
 2143728.7812128419800.7477763642143149.08591155420259.312716156
#Sta/Elev= 30
       0 3477.36    12.4 3476.21    24.9 3468.35    36.1 3463.82   187.7 3411.92
     286  3396.3   317.8 3398.21   393.9 3397.63   402.8 3394.49   420.4 3379.27
  432.71 3376.96   440.2 3376.03   465.8 3377.03   477.5 3380.92     506  3381.1
   521.9 3385.55   531.4 3385.43   538.3 3386.91   543.7 3390.67     552  3398.9
     592 3427.06   606.4 3440.54   615.3 3446.12   631.5 3453.28     662 3464.13
   677.5 3472.91   708.8 3473.91   711.1 3474.65   720.4 3481.63   739.1 3487.84
#Mann= 3 , 0 , 0
       0     .12       0  432.71     .04       0   465.8     .12       0
Bank Sta=432.71,465.8
XS Rating Curve= 0 ,0
Exp/Cntr(USF)=0,0
Exp/Cntr=0.3,0.1

Type RM Length L Ch R = 1 ,75787   ,368.7,365.6,366.5
XS GIS Cut Line= 3
2143675.92653568419755.6162100232143285.19543003419846.483909012
2142980.13958342420060.672056628
#Sta/Elev= 30
       0 3473.04    16.7 3471.19    30.3 3461.99    57.7 3451.76   106.8 3429.34
   147.7 3413.78   184.8 3403.79   194.9 3397.83   211.7 3383.57   225.2 3374.75
   235.3  3366.5   240.8 3364.49     249 3363.82   268.1 3362.88   275.7 3364.06
   289.2 3367.47   326.2  3368.5   339.7 3371.48   356.5 3370.81   393.6 3380.36
   421.4 3383.58   456.3 3390.57   493.7 3395.58   507.1 3398.81   524.5 3400.74
   540.5 3404.45   575.6 3409.95   604.1 3417.06   628.7 3421.24   773.9 3459.41
#Mann= 3 , 0 , 0
       0     .12       0     249     .04       0   275.7     .12       0
Bank Sta=249,275.7
XS Rating Curve= 0 ,0
Exp/Cntr(USF)=0,0
Exp/Cntr=0.3,0.1

Type RM Length L Ch R = 1 ,75421   ,452.9,452.7,456.8
XS GIS Cut Line= 2
     2143687.943      419349.076     2142773.226      419686.944
#Sta/Elev= 30
       0 3573.51    42.5 3548.46    62.2 3538.86   104.7 3512.25   166.9 3482.15
   186.5 3474.77   206.2  3470.8   225.8 3463.04   245.4 3448.38     265 3446.22
     301 3420.99   314.1 3414.23   333.8  3408.8   359.9 3397.84   431.9 3378.99
   464.7 3357.44     481  3348.8   487.6  3348.2   507.2 3349.25   556.3 3357.77
   615.2 3360.89   670.8 3368.73   710.1 3379.42     733 3387.75   746.1 3394.71
   759.2 3396.39   850.8 3432.73     877 3444.95     913 3465.38   975.1 3496.27
#Mann= 3 ,-1 , 0
       0     .12       0     481     .04       0   507.2     .12       0
Bank Sta=481,507.2
XS Rating Curve= 0 ,0
Exp/Cntr=0.3,0.1

Type RM Length L Ch R = 1 ,74969   ,407.4,406.3,408.7
XS GIS Cut Line= 2
2143575.68503261419076.7641152632142555.11069285419149.842277864
#Sta/Elev= 30
       0 3556.23      26 3542.59    50.5 3524.59    63.5 3520.86    86.5 3506.67
   102.9 3501.98   179.4 3462.23   234.5 3437.62   247.7 3433.87   267.4 3419.52
   287.1 3418.62   301.6 3408.13     320 3399.15   408.8 3363.77   435.2 3349.25
   451.6 3344.78   497.7 3342.74     514 3336.66   530.5  3335.9   537.1 3334.84
   550.3 3335.85   556.9  3340.1   576.6 3345.65   632.5  3350.8   711.5 3369.01
   803.6 3401.91   836.4 3419.21   859.5 3427.07   974.6 3478.74  1023.2 3497.34
#Mann= 3 , 0 , 0
       0     .12       0   530.5     .04       0   550.3     .12       0
Bank Sta=530.5,550.3
XS Rating Curve= 0 ,0
Exp/Cntr(USF)=0,0
Exp/Cntr=0.3,0.1

Type RM Length L Ch R = 1 ,74562   ,343.3,339.9,339.7
XS GIS Cut Line= 2
     2143671.461      418742.012     2142520.512      418687.074
#Sta/Elev= 30
       0 3600.65    62.2  3571.2    98.2 3549.31   117.8 3533.44     180  3501.3
   206.2 3484.55   281.5 3455.35   294.6 3446.77   304.4 3444.02   340.4 3418.48
   373.2 3406.76   389.5 3392.04   409.2 3389.99   432.1 3372.86   487.8 3355.53
   520.5 3339.12   536.8  3333.8   556.5 3330.87   592.5  3332.1     622 3327.64
   638.3 3326.41   651.4 3328.23   677.6 3332.73   713.6 3331.48   762.7 3337.77
   890.4 3366.68   975.5 3394.83  1080.2 3442.51  1132.6 3459.17  1152.3 3470.96
#Mann= 3 ,-1 , 0
       0     .12       0     622     .04       0   651.4     .12       0
Bank Sta=622,651.4
XS Rating Curve= 0 ,0
Exp/Cntr=0.3,0.1

Type RM Length L Ch R = 1 ,74222   ,311.8,310.6,313.5
XS GIS Cut Line= 4
2143464.80782039418396.3812220862143147.29580358418371.181855672
2142751.66575088418411.5008419342142514.79170659418434.180271707
#Sta/Elev= 30
       0 3469.71    21.6  3461.2    34.6 3453.68    54.8 3450.34    83.9 3429.86
   123.4 3409.13   179.4 3387.68   202.4 3368.45   225.5 3365.53   245.2  3352.2
   264.9 3342.89   277.4 3343.06   294.6 3340.04   317.6 3323.89   337.4 3321.57
   393.5 3325.21   439.6 3325.53   481.43321.619   505.6 3320.97   508.83321.872
   528.7 3324.09   588.4 3321.18   624.3 3323.26   680.5 3353.39   719.9 3371.66
   841.9  3412.4   861.7 3424.33   874.8 3427.89   937.5 3460.65   954.1 3466.04
#Mann= 3 , 0 , 0
       0     .12       0   481.4     .04       0   508.8     .12       0
#XS Ineff= 2 , 0
          417.66 3332.65  533.11         3332.04
Permanent Ineff=
       F       F
Bank Sta=481.4,508.8
XS Rating Curve= 0 ,0
Exp/Cntr(USF)=0,0
Exp/Cntr=0.3,0.1

Type RM Length L Ch R = 1 ,73912   ,413.4,410.8,396
XS GIS Cut Line= 4
     2143600.042      418269.546     2143223.717      418107.479
     2142729.276      418093.745     2142449.093      418165.164
#Sta/Elev= 30
       0 3483.83    91.8 3456.06   173.7 3416.75   252.4 3392.14     354 3350.02
   373.7 3349.03   455.6 3333.11   481.8 3316.61   606.3 3317.04   668.5 3313.42
   737.3 3317.89   750.4 3313.51   760.2 3313.03   776.6 3313.91   796.3 3328.62
   825.8 3334.35   861.8 3348.34   878.2 3351.67   901.1 3362.88   927.1 3382.01
   940.1 3385.53  1001.8 3415.88  1011.6 3418.05  1040.8    3436  1060.3 3441.92
    1083 3455.23  1141.5  3481.9    1161 3487.22  1180.5 3502.22  1193.5 3506.46
#Mann= 3 ,-1 , 0
       0     .12       0   750.4     .04       0   776.6     .12       0
#XS Ineff= 2 , 0
           736.6 3318.58
Permanent Ineff=
       F       F
Bank Sta=750.4,776.6
XS Rating Curve= 0 ,0
Exp/Cntr=0.3,0.1

Type RM Length L Ch R = 1 ,73501   ,348.5,345.9,347.9
XS GIS Cut Line= 3
2143542.92585628417693.3188991372142880.18251959417768.916998378
2142464.39297376417852.074907544
#Sta/Elev= 30
       0 3431.57    50.6 3418.35    73.7  3408.3   101.2 3401.26   212.4 3356.92
   348.4 3327.58   413.8 3315.86   452.8 3314.56   469.9 3306.94   489.7 3313.06
   501.4 3303.87     536 3301.96   557.1 3303.47   585.5 3308.18   628.8 3308.14
   652.5 3305.06   691.5 3306.66   708.2 3311.17     725 3323.45   776.1 3330.95
   809.5 3350.62   848.6 3369.69   884.8 3394.15   922.4 3412.84   966.1 3443.33
     988    3454  1002.7  3464.7  1056.2 3477.11    1080 3485.59  1091.1 3492.68
#Mann= 3 , 0 , 0
       0     .12       0   501.4     .04       0   557.1     .12       0
Bank Sta=501.4,557.1
XS Rating Curve= 0 ,0
Exp/Cntr(USF)=0,0
Exp/Cntr=0.3,0.1

Type RM Length L Ch R = 1 ,73155   ,150.8,151.7,151.1
XS GIS Cut Line= 4
     2143682.449      417376.805     2143083.626      417409.767
     2142833.658      417464.705     2142369.433      417607.544
#Sta/Elev= 30
       0 3536.65   147.5  3480.5   239.2 3430.75   255.6  3426.2     390 3348.13
   412.9 3346.04   439.2 3331.97   475.2 3323.57   586.6 3315.75     603 3311.25
   619.2 3296.01   661.3 3298.32   674.2 3294.09   687.2 3293.19  701.16 3294.27
   713.1 3299.26   768.2  3301.4   865.4 3294.94   881.7 3298.44     898 3313.69
   917.6 3318.02   982.8 3318.45  1012.1 3336.36    1035  3342.3  1057.8 3357.34
  1080.6 3365.89  1145.8 3406.39  1230.5  3439.3 1319.93 3487.16  1341.4 3487.92
#Mann= 4 ,-1 , 0
       0     .12       0   674.2     .04       0  701.16     .12       0
 1319.93     .08       0
#XS Ineff= 2 , 0
                          805.77         3355.23
Permanent Ineff=
       F       F
Bank Sta=674.2,701.16
XS Rating Curve= 0 ,0
Exp/Cntr=0.3,0.1

Type RM Length L Ch R = 1 ,73003   ,175.8,175.9,175.8
XS GIS Cut Line= 3
2143541.53673403417136.5115996742142745.66332769417337.948541231
2142386.23662805417474.214707579
#Sta/Elev= 30
       0 3496.44    26.7 3490.86   104.5 3442.24   162.1 3422.02   216.2 3387.85
     267  3361.8   307.6 3355.07   341.5 3337.44   422.7 3335.01   507.3 3312.79
   547.9  3292.5   588.5 3292.29   630.73292.689   702.7 3297.86   757.7 3290.39
   776.4 3294.91   798.3 3310.57   864.2 3317.69   923.6 3333.85   948.4 3333.41
   962.4 3342.76   979.9 3348.66     994 3359.61    1013 3363.61  1043.1 3382.66
  1053.7 3385.39  1071.2 3400.32  1102.7 3419.13  1116.8 3422.96  1205.4 3467.34
#Mann= 3 , 0 , 0
       0     .12       0   588.5     .04       0   630.7     .12       0
#XS Ineff= 2 , 0
                           708.4          3302.7
Permanent Ineff=
       F       F
Bank Sta=588.5,630.7
XS Rating Curve= 0 ,0
Exp/Cntr(USF)=0,0
Exp/Cntr=0.3,0.1

Type RM Length L Ch R = 1 ,72828   ,412.2,408.9,410.3
XS GIS Cut Line= 3
2143588.60577885416931.4863761762142992.60577796417097.584737081
2142279.35987525417324.748671847
#Sta/Elev= 30
       0 3537.11    65.5 3503.92     120 3484.87   160.9 3460.85   194.9 3435.81
   240.5 3418.52   291.1 3412.88   365.2 3375.61   409.5 3371.19   464.2 3351.34
   508.3 3349.11     616 3320.92   672.3 3313.55     697 3294.21   710.2 3289.74
   758.4 3287.17     786 3285.98   796.3 3287.41   806.6  3291.1   858.3 3288.51
   896.1 3295.56   909.9 3303.75   930.6 3308.33   989.1 3314.74  1030.4 3324.66
  1075.2 3326.87  1144.1 3358.71  1185.4 3366.06  1263.7 3417.85  1367.3 3470.13
#Mann= 3 , 0 , 0
       0     .12       0   758.4     .04       0   796.3     .12       0
#XS Ineff= 2 , 0
                          809.44         3297.69
Permanent Ineff=
       F       F
Bank Sta=758.4,796.3
XS Rating Curve= 0 ,0
Exp/Cntr(USF)=0,0
Exp/Cntr=0.3,0.1

Type RM Length L Ch R = 1 ,72419   ,381.3,379.7,379
XS GIS Cut Line= 2
     2143361.062      416519.773     2142056.286      417005.974
#Sta/Elev= 30
       0 3494.75    65.5 3466.15   104.8 3441.56   199.8 3398.59   268.7 3359.13
   288.3 3356.15   317.8 3337.92   373.5 3328.95   429.2  3302.1   504.6 3299.49
   547.1 3276.94   671.6 3283.38   727.3 3275.74   733.9 3274.92   753.5 3275.84
     783 3280.73   874.8 3278.69   884.6 3280.98   907.5 3295.46  1077.9 3326.96
  1130.3 3346.76    1209 3364.19  1238.4 3375.67    1281 3406.32  1297.4 3409.25
 1320.05    3429  1336.7  3439.8  1359.7 3440.86 1376.41 3457.98  1392.4 3466.54
#Mann= 5 ,-1 , 0
       0     .12       0   727.3     .04       0   753.5     .12       0
 1320.05     .08       0 1376.41     .12       0
#XS Ineff= 2 , 0
          649.17 3287.01  842.88          3284.5
Permanent Ineff=
       F       F
Bank Sta=727.3,753.5
XS Rating Curve= 0 ,0
Exp/Cntr=0.3,0.1

Type RM Length L Ch R = 1 ,72039   ,362.2,360.4,358.4
XS GIS Cut Line= 3
2143177.53504327416115.8385616222142328.31639512416519.028424246
2141985.60501189416730.703102123
#Sta/Elev= 30
       0 3424.57   112.4  3392.2   186.2 3361.04   199.5  3352.2   218.2 3351.67
   301.2  3329.4   326.7 3330.07   348.4  3319.3   399.3 3307.04   457.4 3303.82
   486.5 3296.45   525.2 3292.86   555.6  3267.9   697.1 3269.21   718.9 3272.32
   740.83266.446   751.6 3266.14   761.83266.479   780.6 3272.19   963.6 3268.12
   990.6 3277.09  1017.6 3278.97  1056.1 3292.06  1098.6 3299.23  1121.7 3307.33
  1183.4 3314.75  1216.3 3327.09  1275.9 3361.07  1295.2  3366.8  1342.9 3392.31
#Mann= 3 , 0 , 0
       0     .12       0   740.8     .04       0   761.8     .12       0
#XS Ineff= 2 , 0
          714.81 3276.26  782.85         3276.04
Permanent Ineff=
       F       F
Bank Sta=740.8,761.8
XS Rating Curve= 0 ,0
Exp/Cntr(USF)=0,0
Exp/Cntr=0.3,0.1

Type RM Length L Ch R = 1 ,71678   ,468,468,470.8
XS GIS Cut Line= 4
      2143300.63      415780.858     2142567.209      415978.634
     2142081.008      416294.528     2141734.899      416536.254
#Sta/Elev= 30
       0 3422.49     203 3378.94   235.7  3364.7     311 3343.37   379.8 3328.21
   396.2 3327.56   425.6 3319.86   533.7  3300.4   576.3 3297.97   595.9 3293.43
   641.8 3294.18   700.7 3287.04   746.5 3275.79   766.2 3263.76   779.3 3259.63
   857.9  3262.7   988.9 3258.26  1015.1 3261.14  1103.6 3261.07  1126.5 3258.66
  1136.3  3257.6  1142.9  3258.7  1188.7 3262.09  1260.8 3261.18  1273.9 3267.07
  1290.3 3282.04  1300.1 3286.32  1480.2  3302.5  1607.8 3319.96  1761.6 3346.38
#Mann= 3 ,-1 , 0
       0     .12       0  1126.5     .04       0  1142.9     .12       0
#XS Ineff= 2 , 0
          880.85 3263.31 1193.62         3262.97
Permanent Ineff=
       F       F
Bank Sta=1126.5,1142.9
XS Rating Curve= 0 ,0
Exp/Cntr=0.3,0.1

Type RM Length L Ch R = 1 ,71210   ,428.3,436.2,436.9
XS GIS Cut Line= 4
2143217.85402954415634.5306631162142454.31322719415637.050599757
2141819.28919356415863.8448974832141463.97812712416072.999638719
#Sta/Elev= 30
       0 3388.12   118.9 3351.08   282.7 3324.75   338.7 3312.19   351.8 3305.94
   374.8 3305.84   522.4 3282.19   706.1 3267.11   748.8 3257.89   779.3 3260.86
     810    3250   883.7 3251.94     936 3248.47   967.4 3252.76   996.1 3247.87
  1069.3 3250.42 1081.13  3247.2  1091.2 3245.56 1109.68 3247.35  1235.6 3248.89
  1305.4 3282.23  1354.2 3295.96  1475.7  3305.8    1585 3321.07  1666.1 3338.21
  1690.5 3339.14    1706 3346.82  1749.8  3354.5  1791.1 3353.61  1850.2 3375.65
#Mann= 3 , 0 , 0
       0     .12       0 1081.13     .04       0 1109.68     .12       0
#XS Ineff= 2 , 0
          964.35 3256.33
Permanent Ineff=
       F       F
Bank Sta=1081.13,1109.68
XS Rating Curve= 0 ,0
Exp/Cntr(USF)=0,0
Exp/Cntr=0.3,0.1

Type RM Length L Ch R = 1 ,70774   ,529.8,523.1,523.1
XS GIS Cut Line= 4
     2143218.223      415558.359     2142410.636      415250.707
     2141726.659      415478.699     2141333.853      415830.302
#Sta/Elev= 30
       0 3379.07    32.7 3365.05      72 3353.61   157.1 3343.07   199.7 3333.56
   219.3 3333.32   261.9 3321.19   422.3  3293.5   474.7 3292.86     563 3282.97
   831.5 3272.42   975.6 3255.87  1034.6 3255.45  1073.9 3251.01  1270.6  3242.1
  1283.7 3235.77  1293.5 3234.79  1313.2 3235.73  1388.6 3239.26    1418 3255.01
  1493.4 3267.93    1559 3285.04  1758.7  3309.2  1935.5 3350.37 1963.48 3353.04
 2003.12 3365.94  2027.2 3367.84  2053.4  3374.8    2096 3393.34  2112.4 3397.07
#Mann= 5 ,-1 , 0
       0     .12       0  1283.7     .04       0  1313.2     .12       0
 1963.48     .06       0 2003.12     .12       0
Bank Sta=1283.7,1313.2
XS Rating Curve= 0 ,0
Exp/Cntr=0.3,0.1

Type RM Length L Ch R = 1 ,70251   ,558.7,555.8,554
XS GIS Cut Line= 3
 2142989.9018044414433.7921584882141813.82408558414899.532337737
2141271.01898458415201.090727179
#Sta/Elev= 30
       0 3421.16    66.2 3403.85    91.2 3393.28   154.4 3382.36   179.1 3373.46
   253.2  3358.8     292 3347.04   380.2 3340.02   419.8 3331.41   616.6 3307.83
   669.6 3295.64   766.1 3278.77   910.2 3264.39   951.9 3252.53  1078.9 3242.24
    1130 3241.45  1160.1 3234.63  1302.7 3231.48  1348.6 3227.47  1423.4 3228.21
  1446.1 3228.24  1483.7 3232.66  1558.5  3233.8  1597.1 3231.54  1645.1 3255.52
  1679.6 3268.36  1713.4 3273.62  1761.4 3290.39  1838.3 3305.84  1885.9 3319.95
#Mann= 3 , 0 , 0
       0     .12       0  1423.4     .04       0  1446.1     .12       0
#XS Ineff= 2 , 0
         1298.25 3233.61 1531.41         3244.32
Permanent Ineff=
       F       F
Bank Sta=1423.4,1446.1
XS Rating Curve= 0 ,0
Exp/Cntr(USF)=0,0
Exp/Cntr=0.3,0.1

Type RM Length L Ch R = 1 ,69695   ,527.3,521.8,521.9
XS GIS Cut Line= 3
      2142699.06      414061.301     2141718.418      414426.638
     2141020.706      414896.357
#Sta/Elev= 30
       0 3473.24    75.4 3435.04   167.3    3409   219.8  3384.3   429.8 3366.86
   472.4 3356.57   524.9 3334.89   547.8 3329.86   751.2 3314.83   803.7 3295.68
   833.2 3309.36   866.1 3309.32   892.3 3302.46   921.8 3285.13   957.9 3271.14
  1026.8 3251.65  1147.9 3233.43  1177.4 3224.73  1301.8 3217.79  1318.1 3216.03
  1334.5 3217.92  1373.8 3221.89  1462.1 3222.21  1478.5 3229.14  1524.3 3260.78
  1573.4 3281.09    1629  3292.4  1717.4  3297.9  1838.5 3323.33  1887.6 3328.02
#Mann= 3 , 0 , 0
       0     .12       0  1301.8     .04       0  1334.5     .12       0
#XS Ineff= 2 , 0
         1285.11 3220.78 1412.77          3222.8
Permanent Ineff=
       F       F
Bank Sta=1301.8,1334.5
XS Rating Curve= 0 ,0
Exp/Cntr=0.3,0.1

Type RM Length L Ch R = 1 ,69174   ,315.7,311.1,315.5
XS GIS Cut Line= 3
2142016.12482912413561.6530613572141238.10418436414104.458162353
2140843.06269419414469.343813577
#Sta/Elev= 30
       0 3427.86    23.8 3415.88    59.8 3408.16   127.8 3375.49   179.8 3361.41
   327.8 3339.59   372.6 3340.97   459.7 3331.19   505.6  3332.8   605.9 3327.92
   635.8 3323.51   651.8 3314.03     719 3312.51   740.2 3303.61   799.9 3286.55
   834.4  3273.6   881.6 3260.93  1000.5 3218.32  1045.1 3211.78  1068.2 3212.19
  1081.8 3209.74  1092.4 3208.84  1111.7 3209.62  1145.6  3213.3  1191.3 3243.89
  1309.5 3278.12  1323.7 3286.34  1348.7    3296  1416.3 3311.37  1486.4 3319.08
#Mann= 3 , 0 , 0
       0     .12       0  1081.8     .04       0  1111.7     .12       0
#XS Ineff= 2 , 0
         1060.54 3212.57
Permanent Ineff=
       F       F
Bank Sta=1081.8,1111.7
XS Rating Curve= 0 ,0
Exp/Cntr(USF)=0,0
Exp/Cntr=0.3,0.1

Type RM Length L Ch R = 1 ,68863   ,426.3,425.9,412.8
XS GIS Cut Line= 3
2141460.18171589413231.1024723232141098.89839961413865.899711663
2140658.01028483414265.964852854
#Sta/Elev= 30
       0  3388.6    49.1 3364.79    71.4  3358.6    82.8 3351.72   135.7 3340.35
   321.6 3329.89   573.5 3300.98   618.8  3299.2     649 3292.59   660.3 3287.06
   699.7 3283.79   720.7 3273.82   740.9 3269.06   820.7 3241.14   842.8 3231.21
   935.8 3204.73   990.1 3206.49  1005.9 3203.53  1033.3 3207.79  1064.3 3204.78
  1094.6 3204.83  1099.3 3207.56  1113.2 3223.21  1126.3 3229.68  1141.1 3231.98
  1223.8  3257.1  1245.6 3272.17  1261.8 3280.15  1290.3 3287.45  1325.8 3301.86
#Mann= 3 , 0 , 0
       0     .12       0  1064.3     .04       0  1094.6     .12       0
Bank Sta=1064.3,1094.6
XS Rating Curve= 0 ,0
Exp/Cntr(USF)=0,0
Exp/Cntr=0.3,0.1

Type RM Length L Ch R = 1 ,68437   ,180.1,184.5,186
XS GIS Cut Line= 3
     2141487.679      413105.381     2140853.146      413649.266
     2140531.759      414129.973
#Sta/Elev= 30
       0 3435.79    13.1 3427.16    26.2 3422.23      36 3414.65    49.2 3411.83
    75.4 3395.36   101.6 3383.33   124.5 3378.41   170.4 3356.67   216.3 3340.87
   301.5 3328.23   416.2 3319.39   599.8 3293.35   701.4 3282.31   724.3 3272.36
   747.2 3270.59   773.5 3255.95   796.4 3254.87   819.3 3242.61   927.2 3202.97
   976.2 3195.51   999.1 3194.49  1008.9 3195.99  1067.7  3202.3  1159.2 3221.81
  1175.5 3223.18  1224.5 3243.04  1312.7  3269.7  1348.6 3286.38    1414 3311.24
#Mann= 3 , 0 , 0
       0     .12       0   976.2     .04       0  1008.9     .12       0
Bank Sta=976.2,1008.9
XS Rating Curve= 0 ,0
Exp/Cntr=0.3,0.1

Type RM Length L Ch R = 1 ,68252   ,283.3,292.8,288
XS GIS Cut Line= 3
2141282.17107105413055.8060195952140799.93963532413465.489363218
2140411.59396585413913.580520306
#Sta/Elev= 30
       0 3359.02    32.2 3348.81    52.5 3347.52    94.5 3336.14   118.3 3326.93
   151.7 3324.44   194.7 3308.05   234.9  3303.9     269 3307.04   332.5 3294.71
   417.3 3286.46   498.4  3283.3   547.7 3276.63     608 3258.52   648.4 3236.07
     674  3236.2   694.9 3225.57   747.7 3208.68   808.5 3201.21   839.1 3194.04
  898.19 3191.26   919.5 3190.19   932.2 3191.29   941.5 3198.21   954.6  3199.3
   969.6 3205.71  1086.4 3228.16  1106.6 3228.33  1119.9 3234.94  1225.7 3258.55
#Mann= 3 , 0 , 0
       0     .12       0  898.19     .04       0   932.2     .12       0
Bank Sta=898.19,932.2
XS Rating Curve= 0 ,0
Exp/Cntr(USF)=0,0
Exp/Cntr=0.5,0.3

Type RM Length L Ch R = 1 ,67959   ,116,111.5,116.1
XS GIS Cut Line= 4
2141211.14114354412776.0753421652140574.05622455413343.911900393
2140401.92458495 413537.807310522140229.79294535413787.101409254
#Sta/Elev= 30
       0 3422.25    72.5 3400.63   134.4 3389.47   214.2 3361.51   251.4 3353.65
   332.8 3328.93   367.3 3313.79     501 3282.78   551.9  3264.6   579.1  3268.1
   602.3 3266.47   713.1 3241.56   771.7 3221.41   796.9 3206.76   846.4  3203.6
   875.2  3205.9   924.63185.736   934.7 3184.27   943.9 3185.34   967.1 3190.44
  1025.2 3190.64  1082.7  3195.5  1134.4 3212.73  1166.3 3215.05  1202.2 3222.41
  1269.2 3246.31  1333.7 3261.43  1385.6 3286.47  1397.5 3287.14  1415.6 3295.86
#Mann= 3 , 0 , 0
       0     .12       0   924.6     .04       0   943.9     .12       0
#XS Ineff= 2 , 0
                          959.64         3198.33
Permanent Ineff=
       F       F
Bank Sta=924.6,943.9
XS Rating Curve= 0 ,0
Exp/Cntr(USF)=0,0
Exp/Cntr=0.5,0.3

Type RM Length L Ch R = 1 ,67848   ,325.9,325.3,325
XS GIS Cut Line= 4
     2141152.557      412685.106     2140476.821      413286.676
     2140377.933       413407.54      2140149.94      413764.636
#Sta/Elev= 30
       0 3443.48    65.6 3427.08   121.3 3403.91   190.1 3386.31   222.9 3371.82
   268.8 3359.98   301.6 3345.13   334.4 3337.71   380.2 3333.29   455.6 3305.07
   491.7 3303.47   668.7 3272.56   757.2 3245.25   806.4 3239.49   816.2 3236.65
   832.6    3222   865.4 3201.16   930.7  3198.1   963.3 3183.34   979.5 3182.84
   989.3 3183.48  1005.6  3187.1  1044.6 3187.62  1168.4 3200.18  1197.8 3210.86
  1279.2 3230.26  1308.6 3242.01  1386.8 3261.58  1458.5 3287.44  1484.6 3292.33
#Mann= 3 , 0 , 0
       0     .12       0   963.3     .04       0   989.3     .12       0
#XS Ineff= 2 , 0
                          1000.9         3200.84
Permanent Ineff=
       F       F
Bank Sta=963.3,989.3
XS Rating Curve= 0 ,0
Exp/Cntr=0.5,0.3

Type RM Length L Ch R = 1 ,67523   ,360.5,359.8,361.5
XS GIS Cut Line= 3
     2140677.344       412451.62     2140056.546      413316.892
     2139913.707      413547.631
#Sta/Elev= 30
       0 3452.48      36 3433.67    81.9  3417.2   108.1 3412.37     154  3393.4
   252.3 3345.72   314.6 3334.53   353.9 3318.44   393.2 3321.76   471.8 3288.59
     639 3260.09   714.3 3235.93   756.9 3217.52   786.4 3216.66   806.1 3208.38
   822.5 3207.34   838.8 3196.22   868.3 3184.17   914.2 3178.94   930.6 3178.18
     947  3179.2   956.8 3183.64   999.4 3186.55  1048.6  3188.6  1064.9 3183.94
    1078 3185.31  1169.6 3212.56  1205.5 3216.15  1297.1 3251.75  1336.3 3259.64
#Mann= 3 ,-1 , 0
       0     .12       0   914.2     .04       0     947     .12       0
#XS Ineff= 2 , 0
          896.19 3192.47
Permanent Ineff=
       F       F
Bank Sta=914.2,947
XS Rating Curve= 0 ,0
Exp/Cntr=0.3,0.1

Type RM Length L Ch R = 1 ,67163   ,457,457.8,446.7
XS GIS Cut Line= 3
2140385.72968453412305.0377920282139674.05188544413218.759712039
2139595.64670419413420.803832966
#Sta/Elev= 30
       0 3400.16    38.2 3386.11      84 3362.32   138.8 3344.23   154.7 3341.24
   229.6 3339.22   316.8 3326.54   370.9 3310.73     454 3292.75     482 3282.56
   503.1 3279.83   526.4 3270.73   571.3 3263.15   636.3 3237.08     662    3236
   763.5 3204.46   827.6 3191.02     845  3178.1   884.1 3174.06     913 3173.53
     9213174.392   940.2 3178.22   966.4 3176.39  1064.1 3178.23  1105.2 3173.83
  1172.8 3177.94  1216.9 3186.81  1318.9  3216.5  1347.1 3220.54  1374.9 3239.79
#Mann= 3 , 0 , 0
       0     .12       0   884.1     .04       0     921     .12       0
#XS Ineff= 2 , 0
                         1071.99         3204.72
Permanent Ineff=
       F       F
Bank Sta=884.1,921
XS Rating Curve= 0 ,0
Exp/Cntr(USF)=0,0
Exp/Cntr=0.3,0.1

Type RM Length L Ch R = 1 ,66705   ,565.9,547.8,531.3
XS GIS Cut Line= 4
     2140180.156      411915.975     2139515.407      412709.828
      2139389.05      412962.542     2139218.742      413374.577
#Sta/Elev= 30
       0 3430.95      59 3406.99   245.8 3351.23   262.1 3344.08   281.8 3340.77
   324.4 3327.51   409.6  3309.7     580  3279.8   635.7 3262.68   668.4 3262.26
   756.9 3249.73   796.2 3239.88   842.1 3232.44     947 3203.43  1022.3 3193.21
  1064.6 3180.42  1106.9  3185.1  1132.8 3170.99  1181.6 3169.48  1194.6 3165.42
    1201 3164.52  1220.5 3165.76    1240 3172.04  1462.2 3166.19  1491.7 3173.86
  1501.6  3181.1  1521.2 3188.13  1596.6  3210.3  1685.1 3230.65  1763.8 3241.38
#Mann= 3 , 0 , 0
       0     .12       0  1194.6     .04       0  1220.5     .12       0
#XS Ineff= 2 , 0
                         1314.09          3185.2
Permanent Ineff=
       F       F
Bank Sta=1194.6,1220.5
XS Rating Curve= 0 ,0
Exp/Cntr=0.3,0.1

Type RM Length L Ch R = 1 ,66157   ,513.3,526,541
XS GIS Cut Line= 4
     2139276.427      411589.094     2138941.306      412627.421
     2138977.016      412797.729     2138908.343      413253.713
#Sta/Elev= 30
       0 3373.75    49.2 3362.84    81.9 3349.22   131.1 3341.09   196.6 3310.51
   258.8 3308.56   294.9 3288.54   363.7 3263.06     403 3260.87   425.9 3264.39
   507.8 3252.76   573.4 3249.55     616 3240.94   638.9 3224.84   658.6 3217.84
   684.8 3228.94   701.2 3230.26   855.2 3200.18   969.8 3162.26    1104  3163.7
  1149.1 3158.69    1162 3157.56  1187.7 3159.22  1258.6 3163.76    1301 3159.49
    1373 3164.09  1402.4 3158.48  1451.5 3162.35  1477.7 3172.26  1726.2 3236.92
#Mann= 3 ,-1 , 0
       0     .12       0  1149.1     .04       0  1187.7     .12       0
#XS Ineff= 2 , 0
         1091.49 3163.51    1260         3164.36
Permanent Ineff=
       F       F
Bank Sta=1149.1,1187.7
XS Rating Curve= 0 ,0
Exp/Cntr=0.3,0.1

Type RM Length L Ch R = 1 ,65631   ,446.4,449.4,442.9
XS GIS Cut Line= 4
2138909.79265652 411691.305277762138630.43733073412471.856923374
2138486.65150127412829.2674137342138416.81266982413108.622739533
#Sta/Elev= 30
       0 3282.42    88.2 3270.94   143.8 3265.89     210 3254.76   262.2 3250.79
   356.3 3251.88   464.3  3242.2   517.3 3235.15   582.8 3222.04   631.6 3214.54
   691.3  3201.8   802.3 3176.61   832.4 3166.91   865.2 3160.57   880.3 3154.37
   963.5 3153.86  1006.4 3150.18  1029.1  3153.5  1079.5 3153.95  1095.5 3153.83
  1106.1 3151.07  1134.4 3151.12  1148.5 3147.99  1169.7 3148.15  1180.3 3150.61
  1229.2 3156.57  1269.9 3169.09  1398.3 3192.06  1421.9 3199.74  1502.2 3211.02
#Mann= 3 , 0 , 0
       0     .12       0  1134.4     .04       0  1180.3     .12       0
#XS Ineff= 2 , 0
            1087 3157.41
Permanent Ineff=
       F       F
Bank Sta=1134.4,1180.3
XS Rating Curve= 0 ,0
Exp/Cntr(USF)=0,0
Exp/Cntr=0.3,0.1

Type RM Length L Ch R = 1 ,65182   ,573.1,577.9,567.5
XS GIS Cut Line= 3
2138326.43300559411913.1462717762138248.37784103412225.366930022
2138047.07767979412989.485909413
#Sta/Elev= 30
       0 3236.47    29.2 3232.65    76.6 3214.36    99.1 3213.93     151 3205.68
   188.2 3189.61   247.9  3175.6   269.3    3168   316.7 3163.12   357.4 3143.72
   391.3 3146.23   499.9 3146.34   520.2 3142.25   581.3 3147.25   614.5 3146.53
   658.53140.878   676.3 3139.28   693.2  3141.3     700 3144.81   720.4 3145.53
   737.3 3153.31   779.4 3154.43     795 3148.18   808.6 3147.26   842.8 3156.79
   869.6 3160.84   940.9 3161.57   981.6 3167.35  1056.3  3171.8    1112 3182.52
#Mann= 3 , 0 , 0
       0     .12       0   658.5     .04       0   693.2     .12       0
#XS Ineff= 2 , 0
          595.96 3151.88
Permanent Ineff=
       F       F
Bank Sta=658.5,693.2
XS Rating Curve= 0 ,0
Exp/Cntr(USF)=0,0
Exp/Cntr=0.3,0.1

Type RM Length L Ch R = 1 ,64604   ,151.1,150.1,147.8
XS GIS Cut Line= 3
     2137754.647      411891.253     2137647.518       412619.18
     2137647.518      413072.418
#Sta/Elev= 30
       0 3212.05    45.8 3195.54    71.9 3191.89   137.3 3171.97   189.7 3158.31
     206 3151.59  238.18 3150.69   284.5 3145.29   323.7  3136.5   359.7 3137.89
   379.3 3133.47     399  3134.9   438.2 3130.92     484 3135.82   503.6  3135.6
   529.8 3134.73   539.6 3131.65   552.6 3130.29   572.3 3131.63     690 3137.91
     739 3145.44     801 3147.05   866.2 3151.73   882.5 3154.46     964 3158.39
   996.6 3161.74  1042.3  3170.7  1110.8 3195.62  1156.4 3207.37    1189 3218.35
#Mann= 4 ,-1 , 0
       0     .12       0  238.18     .12       0   539.6     .04       0
   572.3     .12       0
#XS Ineff= 2 , 0
          485.11 3139.46  607.13         3140.41
Permanent Ineff=
       F       F
Bank Sta=539.6,572.3
XS Rating Curve= 0 ,0
Exp/Cntr=0.3,0.1
