HEC-RAS study SFKCHERRYRV.prj: SFKCHERRYRV

--- SFKCHERRYRV.g01 (geometry) --- (continued)

Type RM Length L Ch R = 1 ,41861   ,439.4,417.7,403.6
XS GIS Cut Line= 4
2126536.68514243423214.4278685282126919.07396211423152.749227391
     2127283.659      423311.0722127546.83047261423235.934065736
#Sta/Elev= 30
       02843.325  60.4812834.173 116.9762819.268 180.1182806.454 219.9972800.504
 253.2292787.858 309.7242758.674 323.0172756.609 375.4522725.326 403.9532726.948
  438.322720.681 461.182 2723.12 471.9132721.848 480.715 2717.82 530.5922716.676
 563.0122717.648 607.8322727.991 647.1772744.306 697.2532743.208 722.2912747.779
 784.8092748.008 803.6472749.932 834.3552756.158 854.8262762.994 868.4742764.458
 899.1812776.661 970.8322809.1071015.1872832.0411032.247 2835.981058.4962847.721
#Mann= 3 , 0 , 0
       0     .12       0 480.715     .04       0 563.012     .12       0
#XS Ineff= 2 , 0
          454.34 2723.92
Permanent Ineff=
       F       F
Bank Sta=480.715,563.012
XS Rating Curve= 0 ,0
Exp/Cntr=0.3,0.1

Type RM Length L Ch R = 1 ,41443   ,336.8,330.7,331.6
XS GIS Cut Line= 3
     2126548.923      423705.541     2127247.525      423567.025
2127542.14601096423526.256330182
#Sta/Elev= 30
       02831.801  22.7832827.642 132.013 2819.06 179.0932804.398 201.4242798.991
 218.9752792.238 232.3542790.282 359.4532744.137 386.2112737.163   392.92732.495
 402.9342719.355   426.62710.269 433.0362708.561 476.5182708.344   496.62710.432
 509.9652713.096 526.6882713.092 558.7052716.176 680.5442715.948 730.5342718.432
 740.4712721.137 757.0312731.169 776.9042734.983 836.5212724.906  849.772729.935
  866.332730.824 879.5792736.936 925.9482744.768 985.5662744.056 1009.632746.958
#Mann= 3 ,-1 , 0
       0     .12       0   426.6     .04       0   496.6     .12       0
Bank Sta=426.6,496.6
XS Rating Curve= 0 ,0
Exp/Cntr=0.3,0.1

Type RM Length L Ch R = 1 ,41113   ,492.5,527.5,633.8
XS GIS Cut Line= 4
2126674.24014159423806.9517257882126966.67723331423965.614403211
2127321.33498284423866.0613507112127626.21620613423894.060646726
#Sta/Elev= 30
       0  2792.8    23.4 2785.28    68.2 2764.75    86.3 2754.68   101.8 2752.18
   142.9 2734.96   172.7 2728.15   284.7 2718.06   356.5 2716.57   380.9 2717.81
   404.7 2712.25     432 2713.76     449 2711.53   460.7 2706.85   472.9 2704.67
   517.2 2704.41   530.8 2706.94   554.7 2708.57   581.9 2706.72     616 2709.85
   674.6 2725.62   707.8 2731.01   770.4 2748.65   786.9  2755.2   829.7 2776.54
     856  2784.9   905.5 2794.73   961.5 2799.88   973.9 2804.22  1007.2 2809.64
#Mann= 3 , 0 , 0
       0     .12       0   460.7     .04       0   530.8     .12       0
#XS Ineff= 2 , 0
                          566.38         2715.31
Permanent Ineff=
       F       F
Bank Sta=460.7,530.8
XS Rating Curve= 0 ,0
Exp/Cntr(USF)=0,0
Exp/Cntr=0.3,0.1

Type RM Length L Ch R = 1 ,40585   ,477.1,471.3,473.4
XS GIS Cut Line= 4
     2126630.226      423847.068     2127151.166      424229.492
     2127262.581      424473.401     2127428.198      424639.018
#Sta/Elev= 30
       0  2802.2    39.4 2782.19      59 2776.79    72.2 2768.74   131.2 2741.13
   147.6 2737.48   170.6 2728.59   206.7 2720.66   272.3 2714.76   288.7 2710.19
   308.4 2714.99   406.8 2711.13   449.4 2706.74   649.5 2705.79   747.6 2699.02
   790.1 2698.13   842.4  2699.5     849  2702.9   862.1 2724.32   881.7 2745.49
   888.2 2750.14     898 2755.49   924.2 2760.95   937.2 2768.31   953.4 2772.12
   979.4 2790.22   992.5 2795.89  1008.7 2801.65  1070.5 2809.64  1148.6 2824.51
#Mann= 3 , 0 , 0
       0     .12       0   747.6     .04       0   842.4     .12       0
Bank Sta=747.6,842.4
XS Rating Curve= 0 ,0
Exp/Cntr=0.3,0.1

Type RM Length L Ch R = 1 ,40114   ,766,750.3,704.2
XS GIS Cut Line= 4
2126514.53049435424122.572826797     2126705.506      424404.143
     2126892.201      424753.444     2127105.998      424994.341
#Sta/Elev= 30
       02793.201  44.3832776.526  76.0972762.088 101.9222747.045 111.7752744.953
 139.7162732.103 246.5612704.655 270.3472701.072 313.9542702.618 337.7392699.287
 367.6532699.581 382.5332695.844 408.036 2693.75 442.0542694.747 456.7572691.601
 477.6372689.045 507.783 2691.61 557.376 2690.87 587.7852697.295 605.7362694.243
 657.8172694.482 672.636 2699.18 686.4412708.729 717.3382723.195 758.9332733.138
 814.8342752.055 849.1682768.081 906.9522781.142 985.9112784.2811058.3772803.142
#Mann= 3 ,-1 , 0
       0     .12       0 456.757     .04       0 507.783     .12       0
#XS Ineff= 2 , 0
          371.35 2699.78  590.04         2699.31
Permanent Ineff=
       F       F
Bank Sta=456.757,507.783
XS Rating Curve= 0 ,0
Exp/Cntr=0.3,0.1

Type RM Length L Ch R = 1 ,39364   ,880.4,862.1,835.5
XS GIS Cut Line= 4
      2125970.77      424852.8142126336.06307643425004.124760122
2126680.03933378425109.562834774 2127027.3828361 425276.81416855
#Sta/Elev= 30
       02918.063  27.3112900.404  76.1052861.476  87.6812841.876 105.436 2821.37
  116.092810.007 133.8932796.203 156.4592770.544 172.9082748.554 189.1022718.533
 204.8692699.181 219.0732690.274  240.382689.609   257.42677.515 304.3012676.816
  325.862678.035 342.2762684.125 434.3862681.924 451.4932679.265 482.3772683.213
 599.0482681.591 691.699 2684.34 707.5352689.781 722.5822689.392 736.4262694.156
 811.6242746.434 901.5742774.599 975.4852788.4861008.2572791.9511140.6782791.048
#Mann= 3 ,-1 , 0
       0     .12       0   257.4     .04       0  325.86     .12       0
#XS Ineff= 2 , 0
                          354.47         2684.97
Permanent Ineff=
       F       F
Bank Sta=257.4,325.86
XS Rating Curve= 0 ,0
Exp/Cntr=0.3,0.1

Type RM Length L Ch R = 1 ,38501   ,314.2,319.2,335.8
XS GIS Cut Line= 4
2125882.17417653425474.1130059832126434.65907377425686.080408398
     2126801.865      425674.8752127182.59016988425851.784829456
#Sta/Elev= 30
       02809.389  83.2642784.625  150.032773.726  202.742762.215  290.592753.769
 448.7212726.484 469.8052719.363 508.4592696.618 561.169 2669.78 602.5742667.827
 622.2682669.567 641.9622667.048 661.6562660.045 707.6092666.286 733.9992662.567
 740.4332660.752 783.1032660.695  806.082663.221 829.0562680.089 897.9862713.141
 959.1282732.7811029.213 2741.761056.5092753.0011079.8612766.4891094.332 2770.67
 1112.422773.2561220.9522775.3521293.3072786.5611336.7192787.8161378.9482800.208
#Mann= 3 , 0 , 0
       0     .12       0 733.999     .04       0  806.08     .12       0
#XS Ineff= 2 , 0
          623.56 2671.64
Permanent Ineff=
       F       F
Bank Sta=733.999,806.08
XS Rating Curve= 0 ,0
Exp/Cntr=0.3,0.1

Type RM Length L Ch R = 1 ,38182   ,527.6,531.5,534
XS GIS Cut Line= 4
2125875.94842217425723.0539074012126373.03657543425940.786734862
2126693.47356679426031.1663990912127063.20855682426179.060395103
#Sta/Elev= 30
       0 2805.84    59.4 2778.63     106  2763.3   184.2 2750.44   224.2 2738.74
   252.8 2723.46   273.9 2721.74   317.3    2705   356.7 2695.65   453.4 2686.71
   498.1 2665.05   621.4 2664.59   679.3 2654.63   690.2 2655.48   731.7 2653.97
   747.5 2655.96   775.7 2662.15   822.5 2658.65   873.6 2664.57   926.5 2661.51
   972.5 2677.43  1018.4 2686.18  1054.5 2699.92  1082.2 2706.15  1124.4 2723.95
  1153.5 2725.87  1184.5 2734.39  1202.2 2743.83  1223.4 2745.83  1273.8 2761.57
#Mann= 3 , 0 , 0
       0     .12       0   690.2     .04       0   747.5     .12       0
#XS Ineff= 2 , 0
                          790.05          2667.1
Permanent Ineff=
       F       F
Bank Sta=690.2,747.5
XS Rating Curve= 0 ,0
Exp/Cntr(USF)=0,0
Exp/Cntr=0.3,0.1

Type RM Length L Ch R = 1 ,37651   ,379.8,372.1,370.2
XS GIS Cut Line= 4
     2125660.615      426102.468     2126314.048      426445.746
     2126551.934      426560.173     2126904.246      426770.958
#Sta/Elev= 30
       0 2822.84   344.4 2690.59   387.1 2681.57   406.8 2668.98   449.4 2650.62
     479 2650.35   505.2 2654.63  560.84 2652.11     620 2650.76   659.4 2653.86
   744.6 2650.45   767.4 2652.87     800 2647.89  812.71 2648.78  820.47 2649.18
   865.2 2651.02   901.1 2651.19  943.81 2654.08  1044.4 2653.59    1077 2658.75
  1119.4 2656.59  1158.5 2661.91  1204.1 2661.61  1243.2 2666.29    1253 2671.12
  1275.8  2690.4  1295.3 2699.52  1334.4  2708.9  1373.5  2726.9  1412.6 2738.74
#Mann= 7 ,-1 , 0
       0     .12       0  560.84     .12       0  812.71     .12       0
  820.47     .08       0   865.2     .04       0   901.1     .12       0
  943.81     .12       0
#XS Ineff= 2 , 0
          578.61 2666.79  920.85         2657.23
Permanent Ineff=
       F       F
Bank Sta=865.2,901.1
XS Rating Curve= 0 ,0
Exp/Cntr=0.3,0.1

Type RM Length L Ch R = 1 ,37279   ,504.9,512.5,526.4
XS GIS Cut Line= 3
2125660.27907634426290.1829667622126336.88563473426810.461656067
2126967.08235699426961.904279245
#Sta/Elev= 30
       0 2779.04    58.1 2768.93    92.4 2757.39   146.2  2734.6   212.5  2723.2
   296.7 2686.89   357.3 2651.88   376.3 2648.49   406.4 2648.18   419.4  2644.7
   551.8 2644.68   584.5 2644.15   622.2 2644.62     650 2648.16   664.7 2646.13
   713.2 2647.03   734.7 2649.28  1015.8 2655.09  1029.3 2657.96  1071.2 2658.48
  1100.2 2656.01    1117 2658.53  1130.5 2668.32  1137.3 2669.42  1282.4 2669.32
  1386.8 2674.23  1397.7 2672.37  1461.2 2674.78  1478.1 2678.99  1501.7 2679.79
#Mann= 3 , 0 , 0
       0     .12       0   551.8     .04       0   622.2     .12       0
Bank Sta=551.8,622.2
XS Rating Curve= 0 ,0
Exp/Cntr(USF)=0,0
Exp/Cntr=0.3,0.1

Type RM Length L Ch R = 1 ,36766   ,504.8,500.7,506.5
XS GIS Cut Line= 2
2125320.59536623426445.1262854072126257.22852495427545.670246901
#Sta/Elev= 30
       0 2798.45      19 2790.59    57.2 2764.88   100.4 2747.54   146.1 2733.53
   225.2 2717.65   247.4 2708.68   319.2 2667.06   341.6 2650.76   358.7 2644.04
   405.3 2638.95   505.3 2640.13     517 2635.24   578.5 2633.24   595.7 2634.54
   608.7 2638.75   699.1 2637.65   723.2 2644.89   772.4  2641.8  1077.9 2648.12
  1102.8  2651.5  1129.9 2647.29  1168.7 2651.07  1238.5 2669.56    1275 2685.75
    1299 2689.17  1315.3 2699.08  1350.9 2709.57  1411.6 2716.93  1445.2 2725.87
#Mann= 3 , 0 , 0
       0     .12       0     517     .04       0   595.7     .12       0
Bank Sta=517,595.7
XS Rating Curve= 0 ,0
Exp/Cntr(USF)=0,0
Exp/Cntr=0.3,0.1

Type RM Length L Ch R = 1 ,36265   ,730.9,708.7,699.7
XS GIS Cut Line= 3
     2125118.596      426942.597     2125522.099      427442.458
      2126046.05      427996.522
#Sta/Elev= 30
       0 2722.79      36 2703.02    85.2 2682.97   170.4  2667.5   232.7 2640.12
   258.9 2635.86  318.36 2632.77   360.5 2631.73   376.9 2626.68     413 2624.87
   439.2 2626.97   445.8  2631.6  458.48 2630.86     472 2629.74   488.4  2635.3
   498.2 2635.62   681.7 2632.92   753.7 2637.15   773.3 2633.23   838.8 2633.69
   887.9 2637.73   979.5 2634.09  1074.4 2635.76    1117 2660.13  1192.2    2716
  1231.5 2727.93    1261 2747.64  1280.6 2752.78    1297 2762.89    1405 2814.32
#Mann= 5 ,-1 , 0
       0     .12       0  318.36     .12       0   376.9     .04       0
   439.2     .04       0  458.48     .12       0
#XS Ineff= 2 , 0
                          452.77         2633.36
Permanent Ineff=
       F       F
Bank Sta=376.9,439.2
XS Rating Curve= 0 ,0
Exp/Cntr=0.3,0.1

Type RM Length L Ch R = 1 ,35557   ,741.9,775.9,806.5
XS GIS Cut Line= 4
2124483.83965285427486.307174171 2124949.2075378427799.034392852
2125570.93903208 427977.735660672125961.84805543428253.233448556
#Sta/Elev= 30
       0 2724.98    46.9 2700.76    82.6 2699.79   122.5 2688.75   150.9  2687.3
   169.8 2673.89   205.2 2661.07   276.3 2624.68   401.5 2622.97   430.5 2628.49
   454.2 2620.62   481.9 2629.62   608.7 2621.37   639.4 2625.81   752.1 2625.64
   786.2 2619.13   822.3 2624.07     892 2621.38   994.4 2622.43  1018.3 2627.54
  1052.5 2620.77  1066.1  2627.2  1168.5 2629.95  1202.7 2649.85  1345.8 2715.96
  1364.6 2718.42  1396.3 2739.14  1442.3 2758.55  1522.4 2782.78  1685.8 2862.41
#Mann= 3 , 0 , 0
       0     .12       0     892     .04       0   994.4     .12       0
#XS Ineff= 2 , 0
          712.05  2666.2
Permanent Ineff=
       F       F
Bank Sta=892,994.4
XS Rating Curve= 0 ,0
Exp/Cntr(USF)=0,0
Exp/Cntr=0.3,0.1

Type RM Length L Ch R = 1 ,34781   ,1254.1,1252.7,1268.4
XS GIS Cut Line= 2
     2124266.422       427520.75     2125214.955      428866.763
#Sta/Elev= 30
       0 2751.03    52.5 2734.81   121.4 2701.18  173.89 2701.33   232.9 2665.92
   262.4 2663.17  282.29 2653.79   318.2 2627.86   337.9  2618.4  462.96 2617.63
   826.6 2619.27   980.8  2616.4  1010.3 2610.61  1033.3 2613.01  1062.8 2609.05
  1082.5 2609.18  1092.3 2612.84  1131.7 2612.22  1148.1 2616.22    1171 2611.44
  1180.9 2607.61  1210.4    2611 1221.76 2610.96  1266.2 2610.68 1294.03 2632.89
  1354.7 2668.46  1377.7 2670.68  1407.2 2682.84  1538.4 2714.38  1646.6 2735.67
#Mann= 8 ,-1 , 0
       0     .12       0  173.89     .12       0  282.29     .12       0
  462.96     .12       0    1171     .04       0  1210.4     .12       0
 1221.76     .04       0 1294.03     .12       0
#XS Ineff= 2 , 0
          972.77 2623.24
Permanent Ineff=
       F       F
Bank Sta=1171,1210.4
XS Rating Curve= 0 ,0
Exp/Cntr=0.3,0.1

Type RM Length L Ch R = 1 ,33528   ,891.4,905.8,923.3
XS GIS Cut Line= 2
     2123233.576      427861.017      2124037.57      429426.849
#Sta/Elev= 30
       0 2743.03    45.9 2713.47    62.3 2706.99    95.1  2702.9   157.3 2671.06
     177 2664.74   245.8 2626.91   285.2 2610.54   511.3  2600.5  740.15 2602.62
   773.6 2600.93     790 2605.81   875.2 2600.96   891.6 2593.72   904.7 2592.93
   960.4 2594.32   986.6 2598.99  1176.7  2600.1  1199.7 2593.68  1307.8 2594.86
  1343.9 2599.04  1383.2 2595.52  1448.8 2595.96  1520.9 2594.62 1537.01 2607.23
  1632.4  2691.2  1658.6 2696.46  1681.5 2715.67 1718.14  2731.9  1760.2 2753.61
#Mann= 6 ,-1 , 0
       0     .12       0  740.15     .12       0  1383.2     .04       0
  1448.8     .12       0 1537.01     .12       0 1718.14     .06       0
#XS Ineff= 2 , 0
         1161.81 2601.68
Permanent Ineff=
       F       F
Bank Sta=1383.2,1448.8
XS Rating Curve= 0 ,0
Exp/Cntr=0.3,0.1

Type RM Length L Ch R = 1 ,32622   ,711.5,711.1,716.6
XS GIS Cut Line= 4
     2122568.097      428345.823     2123028.813      429204.019
     2123055.914      429387.703     2123131.194      429631.612
#Sta/Elev= 30
       0 2642.66     6.6 2635.96    49.2 2630.16   101.7 2608.46   180.4 2609.63
   219.7 2602.22   278.8 2599.18   301.7 2592.36  599.34 2589.17     633 2583.82
     692 2587.15   783.8 2582.33   796.9 2586.22   869.1 2588.28   888.8 2581.64
   967.5 2586.78  1003.4 2587.04 1011.99 2582.69  1029.4 2579.99  1068.5 2583.08
 1088.17 2582.91  1101.1  2587.4  1117.4  2587.3  1136.9  2606.8  1159.7 2621.62
  1185.9 2633.62  1267.7  2646.4  1316.8 2657.81    1343 2659.01    1415 2685.17
#Mann= 5 ,-1 , 0
       0     .12       0  599.34     .12       0 1011.99     .04       0
  1068.5     .12       0 1088.17     .12       0
#XS Ineff= 2 , 0
          728.19 2590.74
Permanent Ineff=
       F       F
Bank Sta=1011.99,1068.5
XS Rating Curve= 0 ,0
Exp/Cntr=0.3,0.1

Type RM Length L Ch R = 1 ,31911   ,651,623.7,569.6
XS GIS Cut Line= 4
     2121962.843      428851.707     2122342.256      429333.501
     2122363.334      429508.152     2122658.434      429824.329
#Sta/Elev= 30
       0 2648.74    52.5 2639.66    78.7 2631.23   118.1 2610.93   131.2 2599.68
     141 2595.03   209.9  2592.3     305 2580.41  479.37 2577.54   554.2  2573.7
   590.3 2574.17   603.4 2578.32   649.1  2575.8     724 2573.94     737 2576.28
  745.31 2577.84   838.3 2577.74   890.7 2575.21   907.1  2579.4   926.8 2597.16
   966.1 2620.99   985.8 2625.39  1034.9 2621.56    1071 2632.68 1093.23 2645.75
    1107 2654.18 1133.63 2660.57  1152.9 2668.69 1180.23 2675.43  1221.7    2685
#Mann= 8 ,-1 , 0
       0     .12       0  479.37     .12       0   649.1     .04       0
     737     .12       0  745.31     .12       0 1093.23     .06       0
 1133.63     .12       0 1180.23     .06       0
#XS Ineff= 2 , 0
          465.65 2581.34  787.89          2584.6
Permanent Ineff=
       F       F
Bank Sta=649.1,737
XS Rating Curve= 0 ,0
Exp/Cntr=0.3,0.1

Type RM Length L Ch R = 1 ,31288   ,648.8,634.1,638.4
XS GIS Cut Line= 2
     2121354.861      429374.378     2122412.935      430111.957
#Sta/Elev= 30
       0 2669.68    91.7 2650.69   137.5 2635.31   163.7 2621.23   255.3 2612.12
   271.7 2608.64   386.3 2602.08   458.3 2591.74   530.3 2587.38   543.4 2583.43
   569.6 2581.54     586 2572.38   605.6 2571.76   615.4 2568.84     622  2565.8
     694 2565.12  709.15  2568.8  725.92 2571.83   851.1 2569.63   893.7 2565.33
   936.2 2568.55   975.5 2582.96  1011.5 2590.88 1122.52 2624.65  1142.5 2627.15
 1158.53 2632.68  1191.6 2639.73    1221 2651.27  1247.2 2653.47  1289.8 2676.39
#Mann= 6 ,-1 , 0
       0     .12       0   615.4     .04       0  709.15     .12       0
  725.92     .12       0 1122.52     .06       0 1158.53     .12       0
#XS Ineff= 2 , 0
                          764.35         2575.31
Permanent Ineff=
       F       F
Bank Sta=615.4,709.15
XS Rating Curve= 0 ,0
Exp/Cntr=0.3,0.1

Type RM Length L Ch R = 1 ,30653   ,361.7,359.8,353.5
XS GIS Cut Line= 2
     2120981.681      429929.758     2122107.806      430594.896
#Sta/Elev= 30
       0 2616.41    85.2  2606.5   265.5 2591.09  405.19 2584.61   419.6  2581.3
     436 2569.33   445.8 2565.39   521.2 2566.05   542.4 2562.27   547.4 2559.79
   570.4 2557.28   619.5 2559.87     672  2565.4   832.6 2564.14   852.3 2560.18
   894.9 2561.11   911.3 2556.36   924.4 2556.63     944 2560.55   993.2 2561.85
  1012.9 2577.09  1058.8    2605  1088.3 2611.92  1130.9 2625.47  1183.3 2647.32
  1212.8 2664.56  1248.9 2667.04  1255.4  2668.9    1298 2700.88  1307.9 2706.21
#Mann= 5 ,-1 , 0
       0     .12       0  405.19     .08       0   542.4     .08       0
   547.4     .04       0   619.5     .12       0
#XS Ineff= 2 , 0
                          767.49         2571.26
Permanent Ineff=
       F       F
Bank Sta=547.4,619.5
XS Rating Curve= 0 ,0
Exp/Cntr=0.3,0.1

Type RM Length L Ch R = 1 ,30294   ,288.1,278.2,275.1
XS GIS Cut Line= 3
2120516.19401048430154.7401597622121437.62242267430597.025797611
2121916.76519701430814.817967764
#Sta/Elev= 30
       0 2629.84    41.4 2616.32   175.6 2597.28   226.5  2600.2     292 2591.39
   332.1 2588.64   375.7  2588.5   397.6 2590.95   535.2 2581.45   568.6 2575.57
   592.2 2562.86   819.7 2561.35   837.9 2557.52   906.9  2557.8   939.8  2560.6
   994.4 2561.07  1099.6 2556.83  1167.7 2556.85  1234.4 2552.27  1286.6 2556.29
  1326.2 2552.58  1340.6 2555.33  1359.5 2554.34  1369.5 2556.11  1401.9 2589.62
  1434.3 2615.35  1490.8 2651.11  1513.6 2668.04  1537.9 2670.83  1548.4 2680.14
#Mann= 3 , 0 , 0
       0     .12       0   837.9     .04       0   906.9     .12       0
#XS Ineff= 2 , 0
          808.69 2564.49  995.31          2565.7
Permanent Ineff=
       F       F
Bank Sta=837.9,906.9
XS Rating Curve= 0 ,0
Exp/Cntr(USF)=0,0
Exp/Cntr=0.3,0.1

Type RM Length L Ch R = 1 ,30015   ,165.9,168.4,166.7
XS GIS Cut Line= 2
     2120421.911      430544.407     2121853.165      430998.808
#Sta/Elev= 30
       0 2592.01    62.3 2587.63   209.6 2568.99   219.7 2567.96   239.4 2576.07
   278.7 2560.08  335.93 2557.01   432.8 2556.42     518 2560.24   642.6 2556.61
  767.41 2558.93   783.6 2558.97   793.4 2555.29   875.4 2555.43  891.36 2556.98
   908.2 2558.46   944.3 2553.76    1000 2556.85  1147.6 2556.18  1206.6 2550.76
  1268.9 2551.29  1288.5 2555.84  1324.6 2596.54  1396.7 2648.43  1409.8 2660.27
  1419.7 2664.62  1455.8 2666.66  1468.9 2676.64  1488.5 2696.77  1501.7 2704.18
#Mann= 7 ,-1 , 0
       0     .12       0   209.6     .08       0  335.93     .12       0
  767.41     .12       0   793.4     .04       0   875.4     .12       0
  891.36     .12       0
#XS Ineff= 2 , 0
          776.91 2565.48
Permanent Ineff=
       F       F
Bank Sta=793.4,875.4
XS Rating Curve= 0 ,0
Exp/Cntr=0.3,0.1

Type RM Length L Ch R = 1 ,29847   ,543.4,495.8,489.1
XS GIS Cut Line= 3
2120166.42512367430639.8433491522121295.61483952430993.195233024
 2121698.8968809431142.985705535
#Sta/Elev= 30
       0 2590.22      82 2586.72     137 2588.95   253.9 2580.21   295.2 2574.38
   326.1 2558.48   339.8 2557.61   583.9 2556.52   625.2 2553.58   687.1 2553.91
     718 2555.48   728.3 2558.44   800.1 2553.77   955.2 2558.14  1024.62554.188
  1111.12553.606  1215.6 2554.95  1238.6 2553.99  1248.8 2550.75  1266.1 2553.48
  1284.5 2551.72  1294.1 2554.91    1353 2554.95  1371.1 2553.78  1390.7 2547.55
  1465.6 2552.57  1472.6  2557.8  1519.3 2612.91    1595 2663.83  1613.4 2667.86
#Mann= 3 , 0 , 0
       0     .12       0  1024.6     .04       0  1111.1     .12       0
#XS Ineff= 2 , 0
          953.48 2578.93 1360.09         2567.24
Permanent Ineff=
       F       F
Bank Sta=1024.6,1111.1
XS Rating Curve= 0 ,0
Exp/Cntr(USF)=0,0
Exp/Cntr=0.3,0.1

Type RM Length L Ch R = 1 ,29351   ,326.6,317.6,317.9
XS GIS Cut Line= 3
2120216.35528118431027.7622651422121149.66514836  431288.9353967
 2121591.3550032431407.999618439
#Sta/Elev= 30
       0 2591.79    80.5 2586.52   121.4 2556.09   128.2 2553.34   233.8 2553.57
   281.5 2550.42   400.8 2551.97   441.7 2549.68     469 2551.56   543.9 2548.24
     629 2554.24   687.1 2551.72   727.8  2554.3   782.4 2548.12   840.3 2554.23
   867.5 2548.12  1003.7  2552.7  1095.1 2545.64  1131.6  2548.7  1255.2 2545.72
  1286.8  2543.8 1300.04  2545.8  1306.1 2551.45  1319.7 2573.94  1340.1 2593.07
    1352  2607.3  1374.1 2627.02  1403.1  2658.6  1408.2 2661.39  1426.6 2662.82
#Mann= 3 , 0 , 0
       0     .12       0  1255.2     .04       0 1300.04     .12       0
#XS Ineff= 2 , 0
          835.22 2564.01
Permanent Ineff=
       F       F
Bank Sta=1255.2,1300.04
XS Rating Curve= 0 ,0
Exp/Cntr(USF)=0,0
Exp/Cntr=0.3,0.1

Type RM Length L Ch R = 1 ,29034   ,336.2,344,342.2
XS GIS Cut Line= 2
      2120281.42      431418.087     2121624.867      431725.411
#Sta/Elev= 30
       0 2570.98      72 2565.45    98.2 2557.34   212.8 2553.41   232.4 2549.35
     419 2544.83   438.6 2548.05   481.2 2548.17   556.5 2544.01   631.8 2547.88
   684.2 2547.45   703.8 2543.89     802 2548.86   900.2 2548.28   952.6 2547.59
   972.2 2541.17  1001.7 2542.45  1060.6 2540.25 1078.86 2542.84  1090.1 2558.44
  1099.9 2567.86  1132.6 2586.54  1152.3  2602.2    1185 2621.84  1201.4  2634.4
  1227.6 2637.34  1253.8  2656.6  1358.5  2711.8  1368.3 2713.16  1378.2 2719.93
#Mann= 3 , 0 , 0
       0     .12       0  1001.7     .04       0 1078.86     .12       0
#XS Ineff= 2 , 0
          809.13 2551.04
Permanent Ineff=
       F       F
Bank Sta=1001.7,1078.86
XS Rating Curve= 0 ,0
Exp/Cntr=0.3,0.1

Type RM Length L Ch R = 1 ,28690   ,700.9,672.8,665.8
XS GIS Cut Line= 3
2120037.05123615431649.1295118882120894.81732167431880.324277127
2121554.89512967432041.155418163
#Sta/Elev= 30
       0 2590.85    82.5 2586.84   221.9 2568.16   236.6 2564.15   259.2 2550.27
   269.4 2548.28   412.1 2549.34   605.8 2543.04     633  2544.7   653.4 2539.74
     796 2545.14   865.6 2542.17   928.4 2545.02   945.3 2541.49   958.8 2545.15
  1036.4 2544.89    1104 2542.82  1117.7 2538.54  1134.4 2536.09  1164.7 2537.94
  1232.3 2542.27  1252.5 2559.45  1272.8 2581.74  1299.8 2599.18  1370.7 2633.15
    1391 2635.01  1404.5 2644.95  1455.2 2666.88    1472 2677.23  1567.8 2717.02
#Mann= 3 , 0 , 0
       0     .12       0  1117.7     .04       0  1164.7     .12       0
#XS Ineff= 2 , 0
          955.01 2547.83
Permanent Ineff=
       F       F
Bank Sta=1117.7,1164.7
XS Rating Curve= 0 ,0
Exp/Cntr(USF)=0,0
Exp/Cntr=0.3,0.1

Type RM Length L Ch R = 1 ,28017   ,818.3,797.1,807
XS GIS Cut Line= 2
     2120628.258       432827.39     2121756.578      432397.135
#Sta/Elev= 30
       0  2573.2    19.6 2568.45      72 2539.39  119.41 2534.44   130.9 2532.67
   176.7 2535.73   268.4 2528.99   294.5 2535.51   327.2    2536   369.8 2530.45
   441.8 2535.85   487.6 2532.89   543.2 2536.47   631.6 2532.82   706.9 2532.33
   742.9 2530.86  751.63  2538.6   762.5 2553.46   785.4 2573.45   880.3 2604.16
   903.2 2614.87   926.1  2616.2  1027.6    2659 1099.35 2697.03  1109.4 2697.73
 1130.96  2706.9 1148.34 2713.11 1162.57 2719.93 1194.18 2735.04  1207.6 2742.26
#Mann= 10 ,-1 , 0
       0     .12       0  119.41     .12       0   631.6     .04       0
   706.9     .12       0  751.63     .12       0 1099.35     .06       0
 1130.96     .12       0 1148.34     .06       0 1162.57     .12       0
 1194.18     .06       0
#XS Ineff= 2 , 0
          537.86 2539.79
Permanent Ineff=
       F       F
Bank Sta=631.6,706.9
XS Rating Curve= 0 ,0
Exp/Cntr=0.3,0.1

Type RM Length L Ch R = 1 ,27220   ,734.1,724.6,735.6
XS GIS Cut Line= 2
     2121177.051      433514.479     2122046.341      433009.589
#Sta/Elev= 30
       0 2621.62      95 2580.35   108.1 2578.23   206.3 2537.23     239 2529.41
   268.5 2529.31  279.99  2524.1   320.9 2521.62   383.1 2520.09     406  2521.7
  416.62 2522.08   468.3 2525.94     501 2522.34   527.2  2525.4   569.8 2545.44
   602.5 2548.02     668 2559.95   684.4 2565.79   726.9 2588.66   746.6 2589.49
   756.4 2599.06   766.2 2605.53   805.5 2626.32   828.4 2634.36   841.6 2641.99
   910.3 2663.46     930 2672.53   943.1 2674.54   956.2 2681.43  1005.3 2695.84
#Mann= 5 ,-1 , 0
       0     .12       0  279.99     .12       0   320.9     .04       0
     406     .12       0  416.62     .12       0
Bank Sta=320.9,406
XS Rating Curve= 0 ,0
Exp/Cntr=0.3,0.1

Type RM Length L Ch R = 1 ,26495   ,711.2,654.4,663.6
XS GIS Cut Line= 2
     2121488.766      434126.933     2122340.494      433690.094
#Sta/Elev= 30
       0 2673.31    42.6 2653.17    95.1 2633.62     118 2620.42   131.1 2617.37
   170.5  2597.1   193.4 2578.96   232.8 2533.92   252.4 2519.16  286.93 2517.73
  299.74 2515.07   308.2 2512.04   327.8 2511.22   373.7 2511.28   396.7  2515.1
   406.5 2517.56   452.4 2515.95   458.9 2518.82     472 2532.52   481.9 2536.49
     554 2531.82   573.7 2532.73   603.2 2540.89   629.4 2543.86   655.6 2541.63
   681.8 2543.62   767.1 2559.91   822.8 2576.09   878.5 2581.69   957.2 2599.44
#Mann= 4 ,-1 , 0
       0     .12       0  286.93     .12       0  299.74     .04       0
   396.7     .12       0
Bank Sta=299.74,396.7
XS Rating Curve= 0 ,0
Exp/Cntr=0.3,0.1

Type RM Length L Ch R = 1 ,25841   ,730.5,725.7,716.4
XS GIS Cut Line= 2
     2121680.016      434793.869     2122581.964      434194.984
#Sta/Elev= 30
       0  2698.8    49.2 2680.32    72.2 2663.71     105 2654.36   170.6 2620.86
     187 2615.67   242.8 2588.04     269 2569.55   298.6 2559.79   347.8 2552.49
   400.3 2512.44   436.4 2512.49   459.3 2507.26  466.89  2507.4  503.57 2511.11
  573.25 2510.59  608.71 2510.76   620.1 2510.11   639.8 2507.46  654.32 2509.96
   662.7 2514.48   695.5 2514.68   711.9 2519.82   754.6 2521.64     794 2529.14
   879.3 2553.78     958 2567.92   974.4 2573.66  1000.6  2574.5  1082.7 2603.58
#Mann= 7 ,-1 , 0
       0     .12       0  466.89     .12       0  503.57     .04       0
  573.25     .08       0  608.71     .12       0   620.1     .04       0
  654.32     .12       0
Bank Sta=620.1,654.32
XS Rating Curve= 0 ,0
Exp/Cntr=0.3,0.1

Type RM Length L Ch R = 1 ,25115   ,464.8,481.8,491.7
XS GIS Cut Line= 2
     2122070.979      435247.159     2122835.907      434737.207
#Sta/Elev= 30
       0 2570.82   117.8 2539.75   225.7 2531.21   238.8 2527.36   251.9 2517.14
  281.57 2512.68   330.4 2510.25   343.5 2502.34   353.3 2499.74   382.8 2499.61
   405.7 2502.02  414.14 2504.56  459.06 2507.29  467.39 2507.43  494.56 2508.56
  520.64 2508.88  530.06 2509.03  565.56 2511.48     638  2507.8   654.3 2502.23
   677.2 2504.08   716.5 2534.61   742.7 2549.49   775.4 2564.54     795 2577.32
   814.6 2578.93   847.4  2602.1   873.5 2614.85   899.7 2630.57   919.3 2635.19
#Mann= 11 ,-1 , 0
       0     .12       0  281.57     .08       0   343.5     .04       0
   405.7     .08       0  414.14     .12       0  459.06     .06       0
  467.39     .12       0  494.56     .06       0  520.64     .12       0
  530.06     .06       0  565.56     .12       0
#XS Ineff= 2 , 0
                          570.21         2512.16
Permanent Ineff=
       F       F
Bank Sta=343.5,405.7
XS Rating Curve= 0 ,0
Exp/Cntr=0.3,0.1

Type RM Length L Ch R = 1 ,24633   ,359.5,410.2,453.1
XS GIS Cut Line= 3
2122189.96633281435429.9843507582122528.72324757435457.637976452
    2123123.2762435229.495564472
#Sta/Elev= 30
       0 2554.53   122.1 2529.22   204.4 2518.07   243.9 2513.43   283.4 2511.65
   316.3 2506.56   363.9 2506.22     385 2502.63   450.5 2504.82     481 2497.62
   557.1 2496.25   572.4 2498.16   613.4  2501.7   641.5 2499.15   662.6  2499.2
   680.1 2504.29   683.7 2505.64   703.8 2521.29   722.4 2538.69   746.9 2556.62
   771.5 2577.28   795.9 2578.76   826.4 2593.91   839.1 2601.92     887 2611.11
   902.6 2616.59   912.7 2622.53   929.6 2622.55   940.2 2630.09   976.7 2644.62
#Mann= 3 , 0 , 0
       0     .12       0     481     .04       0   572.4     .12       0
#XS Ineff= 2 , 0
                          619.75         2502.03
Permanent Ineff=
       F       F
Bank Sta=481,572.4
XS Rating Curve= 0 ,0
Exp/Cntr(USF)=0,0
Exp/Cntr=0.3,0.1

Type RM Length L Ch R = 1 ,24223   ,536.6,503.6,499.9
XS GIS Cut Line= 4
2122035.15903099435616.132990824     2122495.939      435689.118
     2122762.247      435859.102     2123124.879      435796.774
#Sta/Elev= 30
       02598.621  12.0982597.621  34.1052586.774 126.7992561.582 173.6182544.968
 259.9832521.903 309.8092516.337 319.7752512.573  426.072504.494 456.5652497.701
 483.023 2495.01 516.4282493.861 548.5522499.222 567.5582491.147 582.5952489.073
 641.5652489.291 648.7632490.846 668.2242496.956 707.1462502.032  765.532503.864
 784.6242502.189 844.5452508.656 974.3742517.1141014.3212532.0991024.3082534.405
1054.2682549.6831077.5712550.8361094.2422562.381 1144.152585.2711150.4082586.618
#Mann= 3 ,-1 , 0
       0     .12       0 567.558     .04       0 648.763     .12       0
#XS Ineff= 2 , 0
          546.14 2501.08
Permanent Ineff=
       F       F
Bank Sta=567.558,648.763
XS Rating Curve= 0 ,0
Exp/Cntr=0.3,0.1

Type RM Length L Ch R = 1 ,23719   ,616.7,542.2,531.7
XS GIS Cut Line= 3
2122042.70630862436094.1614343012122544.81555434436195.597645558
2123133.14557963435962.294359668
#Sta/Elev= 30
       0 2616.33   6.5842611.301   33.362598.532  153.752547.462 160.5512542.634
 167.2452534.771 194.0222488.939 227.4932486.039 234.5032485.292   273.52486.056
 345.8862488.644 362.593    2494  381.462495.344 458.4442493.617 498.6092496.546
 621.3942493.575  649.632490.993 691.9822496.707 731.0932495.367 751.9822498.852
 864.9222505.192 896.6862511.303 918.7212507.164 946.0972507.4781030.8022514.219
1062.5672519.3631090.8022527.834 1101.392533.5611122.5662534.6671145.1532547.625
#Mann= 3 ,-1 , 0
       0     .12       0 227.493     .04       0   273.5     .12       0
#XS Ineff= 2 , 0
                          389.71         2498.62
Permanent Ineff=
       F       F
Bank Sta=227.493,273.5
XS Rating Curve= 0 ,0
Exp/Cntr(USF)=0,0
Exp/Cntr=0.3,0.1

Type RM Length L Ch R = 1 ,23177   ,961.9,969.6,983.2
XS GIS Cut Line= 2
     2122185.588      436815.896     2123185.311      435987.812
#Sta/Elev= 30
       0 2614.19    26.2 2607.93    49.2 2598.46      59 2597.24    98.3 2581.52
     141 2558.84   157.4 2548.08   173.7 2532.88   183.6 2526.71   203.2 2521.72
   252.4 2493.79   278.6 2487.52   285.2 2482.34   311.4 2479.62   399.9 2482.37
   409.8 2486.33   445.8 2484.57   458.9 2487.86   537.6 2485.96   563.8 2491.28
   649.1 2488.64   717.9 2492.33   783.5 2491.88   884.1 2499.35   917.9 2503.74
  1035.9 2507.73  1219.5 2527.99  1242.4 2539.53  1258.8 2543.76  1298.1 2561.38
#Mann= 4 ,-1 , 0
       0     .12       0   285.2     .04       0   399.9     .12       0
   884.1     .12       0
#XS Ineff= 2 , 0
                          428.24         2490.92
Permanent Ineff=
       F       F
Bank Sta=285.2,399.9
XS Rating Curve= 0 ,0
Exp/Cntr=0.3,0.1

Type RM Length L Ch R = 1 ,22208   ,1090.3,1167.1,1231.3
XS GIS Cut Line= 3
     2122387.339       437520.52     2122956.459      437409.105
     2123378.029      437126.051
#Sta/Elev= 30
       0 2536.19    52.4 2515.76    91.7 2504.27   127.8  2496.5   137.6 2492.81
   170.4 2473.38   176.9  2472.3   206.4 2475.43   258.8 2477.16   327.6 2474.92
   347.3 2472.82   376.8 2477.11     521 2477.61   566.8 2476.17   622.5 2478.02
   632.3 2475.06   648.7  2473.2   720.8 2473.22   730.6 2474.93   760.1 2474.96
   789.6 2478.21   815.8 2475.84  827.28 2476.33   845.3 2480.28   858.4 2488.55
   871.5 2500.01     878 2503.34   959.9 2521.92   982.9 2525.41  1087.7 2533.11
#Mann= 4 ,-1 , 0
       0     .12       0   632.3     .04       0   730.6     .12       0
  827.28     .12       0
#XS Ineff= 2 , 0
          262.78 2481.24  796.96         2480.79
Permanent Ineff=
       F       F
Bank Sta=632.3,730.6
XS Rating Curve= 0 ,0
Exp/Cntr=0.3,0.1

Type RM Length L Ch R = 1 ,21040   ,493,485,462
XS GIS Cut Line= 3
     2122297.003      437776.473     2122565.001      437945.101
     2122965.493      438526.266
#Sta/Elev= 30
       0 2563.74    13.1 2561.81    39.2 2549.31    78.3 2537.28   104.5 2523.43
   143.6 2506.97   156.7 2504.69   199.1 2489.01     284 2467.77     333 2465.33
   352.6 2469.43   372.2 2469.33   385.2 2466.46   453.9 2468.94   463.7 2468.16
   473.5 2463.98   506.2  2463.1   561.7 2468.41   617.2    2467   623.8 2464.39
   646.7 2461.52   689.1 2462.37   695.7 2464.55   708.7 2470.55   731.6 2471.26
   754.5 2474.81   757.8 2475.87   767.6 2484.69   774.1 2487.27  1022.4 2517.08
#Mann= 3 , 0 , 0
       0     .12       0   623.8     .04       0   695.7     .12       0
#XS Ineff= 2 , 0
          450.09  2472.2
Permanent Ineff=
       F       F
Bank Sta=623.8,695.7
XS Rating Curve= 0 ,0
Exp/Cntr=0.3,0.1

Type RM Length L Ch R = 1 ,20555   ,746.3,731.8,737.9
XS GIS Cut Line= 2
     2122029.005      438279.346     2122848.055      438830.399
#Sta/Elev= 30
       0 2573.49    62.3 2555.26   124.6 2544.23   150.9 2536.48     164 2530.57
   177.1 2529.31   200.1  2522.5   219.7 2512.75   236.1 2501.68   255.8 2486.04
   272.2  2475.4   285.3  2461.8   288.6 2460.07   321.4 2457.79   341.1 2460.87
     410 2463.44  418.26 2458.44   426.4 2456.39   455.9 2456.14   485.4 2458.42
  510.97 2460.89   541.1 2458.88   564.1 2465.85   590.3 2467.14  611.81 2477.42
   629.7 2487.84   646.1 2491.39   747.8 2503.05   806.8 2507.78   987.2 2533.48
#Mann= 5 ,-1 , 0
       0     .12       0  418.26     .04       0   485.4     .12       0
  510.97     .12       0  611.81     .12       0
#XS Ineff= 2 , 0
          401.94 2467.75
Permanent Ineff=
       F       F
Bank Sta=418.26,485.4
XS Rating Curve= 0 ,0
Exp/Cntr=0.3,0.1

Type RM Length L Ch R = 1 ,19824   ,617.5,650.6,686.5
XS GIS Cut Line= 3
      2121619.48      438845.455     2122032.016      439119.475
     2122450.575      439372.417
#Sta/Elev= 30
       0 2569.54    26.2 2555.01    75.4 2536.14   170.6 2510.31   232.9  2505.3
   252.5 2501.48   275.5 2501.46   331.3 2495.52   419.8 2475.12   511.6  2467.1
   521.3 2464.08   534.4 2457.31   557.2 2450.78   563.7 2448.71   612.6 2447.88
   635.4 2448.46     642 2450.87   658.3 2452.46   677.8  2456.9  710.99 2456.22
   733.3 2461.56   765.9 2463.15   785.4  2471.6   850.6 2478.52     880 2487.82
     906 2499.46   938.7 2509.37   951.7 2517.17   964.7  2520.5   984.3 2529.82
#Mann= 4 ,-1 , 0
       0     .12       0   557.2     .04       0     642     .12       0
  710.99     .12       0
#XS Ineff= 2 , 0
                          692.39         2458.22
Permanent Ineff=
       F       F
Bank Sta=557.2,642
XS Rating Curve= 0 ,0
Exp/Cntr=0.3,0.1

Type RM Length L Ch R = 1 ,19173   ,486.9,492.9,502.2
XS GIS Cut Line= 3
      2121496.02      438875.567     2121730.895      439486.843
     2121779.074      439995.739
#Sta/Elev= 30
       0 2582.01    16.4 2573.49    65.5 2556.86   121.2 2533.99   147.3  2519.6
     167 2515.99   199.7 2502.04   288.1 2473.71     406 2466.54   494.4 2458.58
   533.7 2454.18   556.6 2447.94   566.4 2448.35   576.3 2452.97   586.1 2454.72
     668  2453.9     704 2452.45   743.3 2443.17   753.2 2441.36   792.5 2441.08
   844.9 2442.92     858 2451.74   887.5 2453.45   897.3 2459.58   910.4 2473.04
   936.6 2493.22   946.5 2497.51  1087.4 2522.55  1113.6 2531.76    1166 2541.63
#Mann= 3 , 0 , 0
       0     .12       0   743.3     .04       0   844.9     .12       0
#XS Ineff= 2 , 0
          684.78 2453.97
Permanent Ineff=
       F       F
Bank Sta=743.3,844.9
XS Rating Curve= 0 ,0
Exp/Cntr=0.3,0.1

Type RM Length L Ch R = 1 ,18680   ,1010,987.1,977.1
XS GIS Cut Line= 3
     2121243.078      439065.273     2121276.201       439429.63
     2121212.966      440010.795
#Sta/Elev= 30
       0 2546.99    26.1 2538.08    62.1 2529.39   101.3 2524.36   163.3 2511.64
   231.9 2491.04   258.1  2487.5   303.8 2476.03   329.9  2464.3   356.1 2447.41
   369.1 2442.76   375.7 2442.52   388.7 2446.14     405 2440.62   437.7  2442.9
   476.9  2435.1   496.5 2432.64   532.4 2432.37  566.03 2435.04   578.1 2443.75
   592.2 2444.11     601 2447.48   617.3 2457.25     650 2460.74   672.8 2461.06
   695.7 2464.48   721.8 2463.02   803.5  2471.9     908 2486.98   950.4 2497.96
#Mann= 4 ,-1 , 0
       0     .12       0   476.9     .04       0  566.03     .12       0
   592.2     .12       0
#XS Ineff= 2 , 0
          438.04 2443.25
Permanent Ineff=
       F       F
Bank Sta=476.9,566.03
XS Rating Curve= 0 ,0
Exp/Cntr=0.3,0.1

Type RM Length L Ch R = 1 ,17693   ,824.6,810.3,799.9
XS GIS Cut Line= 2
     2120210.231      439327.249     2120448.117      440170.389
#Sta/Elev= 30
       0 2536.05    26.2 2526.74      36 2521.55    52.3 2519.73    78.4 2509.49
   179.8 2478.45   209.2 2466.69   222.3 2465.01   225.6 2463.67   235.4 2453.78
   245.2 2446.28     255 2440.62     268 2429.87   277.8 2424.64   294.2  2422.6
   323.6 2422.16   362.8 2422.25   369.4 2424.39   379.2  2430.3   382.5 2431.06
   408.6 2431.26  427.58 2441.68   483.8 2454.88   601.5 2476.13   702.8 2501.55
   715.9 2504.07   732.2  2504.7     742 2508.44   853.2    2534   876.1 2541.91
#Mann= 4 ,-1 , 0
       0     .12       0   277.8     .04       0   369.4     .12       0
  427.58     .12       0
Bank Sta=277.8,369.4
XS Rating Curve= 0 ,0
Exp/Cntr=0.3,0.1

Type RM Length L Ch R = 1 ,16883   ,744.1,750.3,764.9
XS GIS Cut Line= 2
     2119343.001      439616.326     2119845.874      440348.051
#Sta/Elev= 30
       0 2516.04    16.4 2515.64    29.5 2509.62    65.5 2500.91      95 2497.04
   124.5 2487.26     154 2482.68   229.3 2463.58   245.7 2462.18   294.9 2452.08
   321.1  2439.6     344 2421.19  356.22 2414.15   363.7 2412.18   396.4  2411.6
   412.8 2414.28  476.56 2415.96     498 2414.74   511.1 2419.43   520.9 2420.61
  548.24 2419.01   648.7 2450.74   681.5 2465.59   727.3 2490.08     747 2493.96
   763.4 2503.28   786.3 2513.38     806 2516.02   871.5 2547.25   887.9 2552.58
#Mann= 5 ,-1 , 0
       0     .12       0  356.22     .04       0   412.8     .12       0
  476.56     .12       0  548.24     .12       0
#XS Ineff= 2 , 0
                          528.26         2422.74
Permanent Ineff=
       F       F
Bank Sta=356.22,412.8
XS Rating Curve= 0 ,0
Exp/Cntr=0.3,0.1

Type RM Length L Ch R = 1 ,16133   ,663.4,662,674.9
XS GIS Cut Line= 3
     2118861.207       439775.92     2119026.824      440360.096
     2119204.486      440781.666
#Sta/Elev= 30
       0 2555.69    16.3 2545.99    42.4 2544.96   58.15    2535    88.1 2526.18
   166.5 2509.03   212.2 2490.26   251.4 2480.94     333 2450.99   385.2 2446.48
     555 2424.46   571.3  2420.7   600.7 2418.79   620.3 2414.16   675.8 2410.43
   698.7  2405.7   731.4 2401.88   760.8 2402.04   770.6 2406.25   777.1 2411.54
   796.7 2412.01  803.23 2415.52   865.4 2461.86   878.4 2477.12     885 2481.69
   914.4  2492.7   973.2 2506.02  1038.5 2524.06  1051.6 2525.69  1064.7 2531.52
#Mann= 5 ,-1 , 0
       0     .08       0   58.15     .12       0   698.7     .04       0
   770.6     .12       0  803.23     .12       0
Bank Sta=698.7,770.6
XS Rating Curve= 0 ,0
Exp/Cntr=0.3,0.1

Type RM Length L Ch R = 1 ,15471   ,785,736.5,677.8
XS GIS Cut Line= 4
     2118301.121      440089.086      2118421.57      440549.802
     2118478.783      440808.767     2118668.489      441179.146
#Sta/Elev= 30
       0 2546.35   101.1 2505.63   185.9 2503.28   231.6 2483.26   313.1 2458.14
   358.8 2446.85   401.2  2444.8   433.8 2432.76   469.7 2428.19   499.1 2407.33
   515.5 2399.66   554.8 2397.14   613.7  2397.3   620.3 2399.39  648.41 2407.49
   666.1 2404.95  708.91 2405.66     725  2415.1   744.7 2419.36   813.5 2420.96
  841.96 2428.61   856.1 2433.42   882.3 2433.78     902 2444.08   924.9 2449.82
   977.3 2456.63  1023.2 2470.03  1042.9 2471.37    1092    2490  1157.6 2521.94
#Mann= 6 ,-1 , 0
       0     .12       0   515.5     .04       0   620.3     .12       0
  648.41     .12       0  708.91     .12       0  841.96     .12       0
Bank Sta=515.5,620.3
XS Rating Curve= 0 ,0
Exp/Cntr=0.3,0.1

Type RM Length L Ch R = 1 ,14734   ,985.6,990.3,1013.8
XS GIS Cut Line= 3
     2117584.452      440968.361     2117897.618      441136.989
     2118400.491      441407.998
#Sta/Elev= 30
       0 2511.58   27.88 2510.39   32.54  2510.2    65.3 2510.73    88.1  2507.9
   107.7 2499.57   150.1 2486.77   195.8 2480.24   234.9 2465.26   274.1 2456.44
     310 2442.66     372 2429.93   427.5  2401.9   453.6 2396.63   466.7 2388.49
     483 2385.49   535.2 2385.52   551.5 2388.38  564.66 2392.78   574.4 2396.28
  631.76 2396.31   685.4 2395.07   744.1 2406.98   796.4 2420.27   845.3 2437.21
   864.9 2445.46     878 2455.05   904.1 2456.26   913.9  2465.1   926.9 2470.01
#Mann= 7 ,-1 , 0
       0     .12       0   27.88     .06       0   32.54     .12       0
   466.7     .04       0   551.5     .12       0  564.66     .12       0
  631.76     .12       0
Bank Sta=466.7,551.5
XS Rating Curve= 0 ,0
Exp/Cntr=0.3,0.1

Type RM Length L Ch R = 1 ,13744   ,578.6,564.8,555.9
XS GIS Cut Line= 4
     2117259.241       441411.01     2117587.463      441956.039
      2117653.71      442175.858     2117870.517      442510.103
#Sta/Elev= 30
       0 2497.99     9.8 2494.08    68.9 2459.48      82 2454.09    98.4 2444.59
   111.5 2442.55   190.2 2403.19   226.3  2393.7   242.7 2392.53   308.3 2381.32
   324.7 2380.98   344.4 2384.18   455.8 2384.48   488.6 2382.43   636.2 2386.05
   662.5 2384.62   685.4  2375.9   731.3 2372.52   760.9 2373.35   767.4 2375.73
   777.3 2381.02   806.8 2381.62   810.1 2383.85  823.88 2402.95   829.7 2409.24
   842.8 2415.24   859.2 2412.44   875.6 2421.66  1078.1 2445.42  1264.2 2479.23
#Mann= 4 ,-1 , 0
       0     .12       0   685.4     .04       0   767.4     .12       0
  823.88     .12       0
#XS Ineff= 2 , 0
          660.43 2386.37
Permanent Ineff=
       F       F
Bank Sta=685.4,767.4
XS Rating Curve= 0 ,0
Exp/Cntr=0.3,0.1

Type RM Length L Ch R = 1 ,13179   ,625.6,629.3,628.6
XS GIS Cut Line= 2
     2116759.379      441787.411     2117412.813      442732.933
#Sta/Elev= 30
       0 2518.52    19.6 2511.08    39.3 2498.97    68.8 2496.99   101.5 2472.28
     131 2465.58   170.3 2452.35   245.6 2400.35   275.1 2386.47     298 2381.25
   327.4 2369.12     370 2368.67   383.1 2371.96     406 2373.03   484.6  2372.3
     537 2367.89   559.9 2361.81   579.6 2359.67   638.5 2361.13   654.9 2371.03
  663.19 2371.65  715.14 2372.94   766.2 2371.82   861.2  2409.8   900.5 2428.17
  1011.8  2455.5  1060.9 2457.08  1070.8 2459.92  1123.2 2459.12  1149.3 2464.14
#Mann= 5 ,-1 , 0
       0     .12       0   559.9     .04       0   638.5     .12       0
  663.19     .12       0  715.14     .12       0
#XS Ineff= 2 , 0
          486.52 2372.05
Permanent Ineff=
       F       F
Bank Sta=559.9,638.5
XS Rating Curve= 0 ,0
Exp/Cntr=0.3,0.1

Type RM Length L Ch R = 1 ,12550   ,559.4,557.3,565.1
XS GIS Cut Line= 2
     2116154.125      442079.499     2117000.276      443118.368
#Sta/Elev= 30
       0 2607.99    65.5 2576.91      95 2566.84   134.3  2547.3   180.2  2529.8
   212.9 2515.03     285 2487.73   363.6 2463.82   412.8 2443.11   422.6  2441.3
     475 2422.11   524.2 2407.34   583.1 2396.34   710.9 2378.73   727.3 2370.38
  742.33  2353.9   763.3 2351.98   845.2 2354.08  853.89 2355.94   881.2 2359.03
   927.1 2357.53  986.75 2358.47 1024.85 2361.42  1123.6 2359.36  1146.6 2361.34
  1159.7 2365.61  1192.4 2382.36  1241.6 2420.73  1287.4 2450.61  1339.9 2467.09
#Mann= 6 ,-1 , 0
       0     .12       0  742.33     .04       0   845.2     .12       0
  853.89     .12       0  986.75     .07       0 1024.85     .12       0
#XS Ineff= 2 , 0
                           881.7         2360.64
Permanent Ineff=
       F       F
Bank Sta=742.33,845.2
XS Rating Curve= 0 ,0
Exp/Cntr=0.3,0.1

Type RM Length L Ch R = 1 ,11992   ,708.8,710.6,718.3
XS GIS Cut Line= 2
     2115694.614      442250.235      2116466.99      443399.315
#Sta/Elev= 30
       0 2701.01    42.6 2683.46    78.6 2657.68   111.3 2639.77   147.3 2623.62
   193.1 2597.66   219.3 2589.18   232.4 2579.94   343.7 2525.83   392.8 2505.61
   487.7 2458.89   510.6 2450.94   569.5 2419.65   648.1 2401.74   674.3 2398.31
   769.2 2402.56   805.2 2392.76   831.4 2380.84   864.1 2362.76   877.2 2352.15
   909.9 2351.45   932.8 2346.51   975.4 2343.93  1021.2 2346.38  1037.6 2350.26
 1072.03 2349.12  1106.3 2355.55  1119.4 2362.25  1214.3 2376.83  1384.5 2412.21
#Mann= 4 ,-1 , 0
       0     .12       0   932.8     .04       0  1021.2     .12       0
 1072.03     .12       0
#XS Ineff= 2 , 0
                         1053.04         2357.79
Permanent Ineff=
       F       F
Bank Sta=932.8,1021.2
XS Rating Curve= 0 ,0
Exp/Cntr=0.3,0.1

Type RM Length L Ch R = 1 ,11282   ,736.7,736.9,726.4
XS GIS Cut Line= 4
     2115152.595      442548.345     2115542.848      443242.129
     2115708.164      443578.181     2115906.001      443887.131
#Sta/Elev= 30
       0 2618.98      36 2595.62   111.4 2555.71   147.4 2530.11   167.1 2525.27
   186.7 2526.19   245.7 2512.36   337.4 2473.67   393.1 2455.47   468.4 2433.24
   599.5 2403.94   674.8 2382.64   753.4 2356.25   828.6 2348.93   848.1 2340.51
  879.64 2338.93  912.56 2343.19     936 2339.95   981.6 2337.57    1024 2340.58
  1046.8  2343.4 1110.06 2340.25    1138 2349.98  1173.8    2352  1229.5 2352.78
  1278.6 2347.65  1393.3 2367.25  1468.6  2385.2    1521 2401.57  1537.4 2402.92
#Mann= 6 ,-1 , 0
       0     .12       0  879.64     .04       0  912.56     .12       0
     936     .04       0    1024     .12       0 1110.06     .12       0
Bank Sta=936,1024
XS Rating Curve= 0 ,0
Exp/Cntr=0.3,0.1

Type RM Length L Ch R = 1 ,10545   ,762.7,802.2,844
XS GIS Cut Line= 3
     2114857.195      442610.677      2115011.67      443710.975
     2115263.709       444152.72
#Sta/Elev= 30
       0 2526.24    26.2 2528.47   108.2 2505.89   144.2 2485.48   190.1 2471.86
   232.7 2455.87   268.8  2446.5   360.5 2410.83     413 2393.32   426.1 2386.72
   547.4 2356.84   599.8 2350.88   760.4 2340.16   816.1 2339.36   852.2 2341.98
     957 2337.98  1065.2 2341.51  1143.7 2341.25  1215.4 2329.83  1251.3 2327.12
  1283.9 2329.88  1293.7 2335.06  1316.5  2333.4    1336  2342.4  1381.7 2346.05
  1414.3 2352.97  1453.4 2354.26  1466.4 2357.96  1525.1 2363.51  1619.7 2369.81
#Mann= 3 , 0 , 0
       0     .12       0  1215.4     .04       0  1283.9     .12       0
#XS Ineff= 2 , 0
                         1298.36         2335.43
Permanent Ineff=
       F       F
Bank Sta=1215.4,1283.9
XS Rating Curve= 0 ,0
Exp/Cntr=0.3,0.1

Type RM Length L Ch R = 1 ,9743    ,644.9,639.3,674
XS GIS Cut Line= 3
     2114769.245      442501.928     2114516.452      443561.429
     2114211.613       444137.65
#Sta/Elev= 30
       0 2562.83   114.5 2521.15   235.5 2469.54   297.7  2451.3   356.5 2427.07
   412.2 2408.22   536.4 2371.33   732.7 2338.49   775.2 2337.23   788.3 2333.76
   860.3 2334.61   889.7 2330.02   951.9 2330.73  1010.7 2336.12  1076.2 2335.76
    1122 2330.79  1207.2 2332.63  1256.3 2329.16  1272.7 2320.61  1334.9 2318.03
  1357.9 2320.46    1371 2322.44  1384.1 2329.92 1414.38  2332.3  1429.9 2345.35
    1443 2345.16  1462.7 2350.62  1534.8 2359.21  1636.3 2393.01  1741.1 2418.62
#Mann= 4 ,-1 , 0
       0     .12       0  1272.7     .04       0  1357.9     .12       0
 1414.38     .12       0
Bank Sta=1272.7,1357.9
XS Rating Curve= 0 ,0
Exp/Cntr=0.3,0.1

Type RM Length L Ch R = 1 ,9103    ,777.5,754.3,754.1
XS GIS Cut Line= 3
     2114613.108        442453.6     2114267.376      443145.064
     2113698.591      443546.559
#Sta/Elev= 30
       0 2540.09    39.3 2519.62      59 2515.48    88.4 2503.64   186.7 2473.72
   219.5 2460.44   291.5 2445.65   327.6  2433.2   363.6 2417.57   448.8 2391.02
   514.3 2382.27   592.9 2359.74   661.7 2344.67   694.5 2340.22   707.6 2334.59
   831.9 2328.72   861.3  2319.1     894 2319.22     930 2323.42  1037.8 2323.61
  1096.7 2313.56  1132.6  2311.2    1198 2313.37  1214.3 2323.34 1238.16 2325.09
  1305.9 2368.23  1335.3 2382.44  1403.9 2399.81  1423.5 2401.98  1469.3 2414.97
#Mann= 4 ,-1 , 0
       0     .12       0  1096.7     .04       0    1198     .12       0
 1238.16     .12       0
#XS Ineff= 2 , 0
         1041.74 2325.68
Permanent Ineff=
       F       F
Bank Sta=1096.7,1198
XS Rating Curve= 0 ,0
Exp/Cntr=0.3,0.1

Type RM Length L Ch R = 1 ,8349    ,418.5,378.6,334.2
XS GIS Cut Line= 4
     2114144.697      442011.212     2113661.416      442639.477
     2113438.363      442914.576     2113237.615      443278.896
#Sta/Elev= 30
       0 2486.07    68.8 2465.03      95 2453.86   170.3 2441.96   219.4 2429.02
   419.2 2389.72   445.4 2389.11   474.9 2378.72   563.4 2367.69   671.4 2349.04
   700.9 2347.32   730.4 2340.14   763.2 2340.73   786.1 2336.91     809 2322.72
   845.1 2306.09   881.2 2303.65   930.4 2303.73   943.5  2306.3   959.9 2311.65
    1055 2312.85  1104.2 2317.38  1130.4 2327.65  1195.9 2333.56  1258.2 2345.02
  1317.1    2352  1425.2 2389.49  1500.5 2421.27  1543.1 2434.35  1562.8 2436.32
#Mann= 3 , 0 , 0
       0     .12       0   845.1     .04       0   943.5     .12       0
Bank Sta=845.1,943.5
XS Rating Curve= 0 ,0
Exp/Cntr=0.3,0.1
